HEC-RAS study SHAVERSFK.prj: SHAVERSFK

--- SHAVERSFK.g01 (geometry) --- (continued)

Type RM Length L Ch R = 1 ,268420  ,533.2,531.6,532
XS GIS Cut Line= 4
2297396.14595984608918.7746326262298060.89194134608811.300731425
  2298749.521012608970.5213257962299115.72837905608890.911028611
#Sta/Elev= 30
       0  3604.2    89.2 3587.16   141.8  3569.6   202.6 3555.98   267.5 3533.36
   320.1 3526.28   397.1 3511.43   416.5 3504.76   441.7 3504.72   474.1 3496.15
     543 3486.28     624 3485.02   771.2 3475.43   832.8    3467   931.3 3463.35
   939.5  3460.6   947.7 3453.88  1062.7 3453.98  1132.5 3461.38  1161.2 3467.66
  1185.8 3465.08  1218.7 3469.04  1276.2  3483.8  1304.9  3481.5  1337.7 3493.03
  1370.6 3498.81    1563 3524.23  1624.4 3540.43  1702.2 3553.48  1754.9 3569.12
#Mann= 9 ,-1,0
       0     .06       0     200      .1       0     300     .06       0
     400     .12       0  803.38      .1       0  903.38     .12       0
   947.7    .045       0  1062.7     .12       0 1103.38      .1       0
Bank Sta=947.7,1062.7
XS Rating Curve= 0 ,0
Exp/Cntr(USF)=0,0
Exp/Cntr=0.3,0.1

Type RM Length L Ch R = 1 ,267888  ,698,642.9,604.1
XS GIS Cut Line= 4
2297424.00956385609464.1051683472297925.55443612609328.767663132
2298470.88497185 609448.183108912299239.12433969609097.897801293
#Sta/Elev= 30
       0 3647.79    70.6 3638.46   103.4 3630.37   134.1 3615.47   223.9  3563.8
   319.2 3538.73   397.9 3511.61   472.5 3491.79   484.9 3485.85   550.8 3476.05
     600  3474.1   661.4 3465.56   821.1 3461.91   853.8 3451.94   968.5 3451.94
  1001.3 3463.81  1029.9 3466.07  1054.5 3477.72  1069.6 3479.82  1290.2 3488.88
  1430.8 3504.08  1461.6 3503.58  1479.2  3507.9  1605.6 3520.26  1681.4 3531.29
  1730.2 3545.57  1817.7 3579.41  1839.7 3578.72    1866 3588.99  1922.1 3601.06
#Mann= 13 ,-1,0
       0      .1       0     380     .12       0  579.48      .1       0
   853.8    .045       0   968.5    .025       0  989.48      .1       0
 1197.74     .12       0 1287.74      .1       0 1297.74     .12       0
 1407.74      .1       0 1627.74     .12       0 1737.74     .06       0
 1847.74      .1       0
Bank Sta=853.8,968.5
XS Rating Curve= 0 ,0
Exp/Cntr(USF)=0,0
Exp/Cntr=0.3,0.1

Type RM Length L Ch R = 1 ,267245  ,767.2,719.3,684.1
XS GIS Cut Line= 2
2297953.41804014610411.4677048572299358.53978547609213.332732213
#Sta/Elev= 30
       0 3704.25    14.9 3693.23    43.3 3677.98    85.9 3656.86   134.1 3638.66
   207.9 3597.91   293.3 3560.88   324.3 3542.16   340.1  3537.7   369.6 3519.33
   484.4 3472.51   497.3 3464.02   518.8 3459.99   529.3 3451.31   534.2 3450.29
   629.2 3450.37   700.2 3462.38   752.6 3464.58   878.9 3464.59   989.9 3474.66
  1012.9 3473.31  1160.1 3481.48  1233.7 3491.54    1465 3514.43  1591.2 3535.27
  1683.3 3564.51  1696.3 3571.26  1723.5 3571.93  1769.9 3589.37  1846.6 3607.19
#Mann= 11 ,-1,0
       0      .1       0   534.2    .045       0   629.2    .025       0
     690      .1       0     710     .12       0     820      .1       0
     860     .12       0    1470      .1       0    1590     .12       0
    1620     .06       0    1720      .1       0
Bank Sta=534.2,629.2
XS Rating Curve= 0 ,0
Exp/Cntr(USF)=0,0
Exp/Cntr=0.3,0.1

Type RM Length L Ch R = 1 ,266526  ,655.5,705,735.2
XS GIS Cut Line= 4
2298650.00814051610702.045289584 2299071.9427156610327.876892812
 2299071.9427156609738.7606936382299497.85780554 609396.43641574
#Sta/Elev= 30
       0 3639.67    50.3 3626.78   127.9 3611.33   155.2 3602.25   291.6 3566.42
   393.2 3550.16   409.2 3544.52   424.3 3529.85   475.3 3507.82   586.6 3470.77
   610.6 3469.18   650.9 3458.78   694.6 3454.96   714.6 3448.16   838.9 3448.11
   854.6  3455.9   870.6 3455.99   898.4 3460.71   926.9 3456.54  1074.9  3464.1
  1219.4 3495.85  1353.5 3508.22  1442.9 3520.02    1584  3551.8  1596.1 3556.18
  1610.1 3565.58  1635.8  3566.4  1647.2 3574.53  1666.5 3583.41  1699.5 3591.63
#Mann= 8 ,-1,0
       0      .1       0     540     .06       0  643.94      .1       0
   714.6    .045       0   838.9    .025       0  843.94      .1       0
 1443.06     .12       0 1523.06     .06       0
#XS Ineff= 2 , 0
                          899.35         3484.48
Permanent Ineff=
       F       F
Bank Sta=714.6,838.9
XS Rating Curve= 0 ,0
Exp/Cntr(USF)=0,0
Exp/Cntr=0.3,0.1

Type RM Length L Ch R = 1 ,265821  ,729.3,756,767.8
XS GIS Cut Line= 2
 2298964.4688144610845.3438245192300238.23356937609810.409961105
#Sta/Elev= 30
       0    3604     9.9 3602.25      32 3592.75    61.5 3589.36   128.5 3572.78
   207.5 3561.88   275.7 3549.15   339.8 3543.86   391.3 3523.95   411.9 3512.05
   458.3 3492.43   477.6  3490.2   514.6 3477.02   545.9 3471.66   618.1  3460.8
   748.8 3458.71   793.2 3452.22   911.9 3454.63   958.1 3446.56  1040.6 3446.53
  1043.5 3446.57  1068.9 3451.31  1087.1 3459.59    1118 3463.01  1211.8 3495.56
  1365.4 3530.99  1521.2 3573.44    1587 3595.53  1617.9 3598.32  1641.2 3608.04
#Mann= 10 ,-1,0
       0      .1       0     330     .12       0     480     .06       0
     510      .1       0     950    .025       0   958.1    .045       0
  1043.5      .1       0    1400     .12       0    1420      .1       0
    1570     .06       0
Bank Sta=958.1,1043.5
XS Rating Curve= 0 ,0
Exp/Cntr(USF)=0,0
Exp/Cntr=0.3,0.1

Type RM Length L Ch R = 1 ,265065  ,431.9,429.8,430.1
XS GIS Cut Line= 2
2299008.25447785611072.2331714982300397.45416374610833.402279941
#Sta/Elev= 30
       0  3632.2      73 3604.79   170.4 3561.11   186.6 3552.08   247.5 3526.21
   304.3 3509.76   365.2  3495.1   377.4 3488.68   397.7 3487.72   450.4 3470.29
   478.8 3464.55   551.9 3460.67   616.8 3453.86   722.4    3456   738.6 3453.08
   742.7  3451.3   746.7 3446.23   750.8 3444.88   884.7 3444.91   909.1 3450.52
   917.2 3454.91   941.5 3458.28  1006.5 3459.39    1043 3482.04  1071.4 3487.82
  1168.8 3513.82  1262.2 3545.19  1314.9 3568.05  1347.4 3576.69  1409.6  3587.6
#Mann= 8 ,-1,0
       0      .1       0     360     .06       0     460      .1       0
   750.8    .045       0   884.7    .025       0     960      .1       0
    1060     .12       0    1160      .1       0
Bank Sta=750.8,884.7
XS Rating Curve= 0 ,0
Exp/Cntr(USF)=0,0
Exp/Cntr=0.3,0.1

Type RM Length L Ch R = 1 ,264635  ,801,800.7,800.5
XS GIS Cut Line= 3
2299155.53352764611498.1482614412300130.75966817611311.064063055
2300512.88909466611151.843468683
#Sta/Elev= 30
       0 3607.67   179.9 3538.86   232.8 3516.12   302.1 3494.64   322.4 3485.73
   338.7 3484.35   346.9 3480.04   363.1 3475.28   425.1 3462.96   497.6 3451.33
   550.5 3450.58   657.5 3455.03   668.6 3454.41   693.1 3448.83   701.2 3443.41
   847.8 3443.43   866.4 3449.74   880.4 3451.46   904.8 3457.96   921.1 3456.97
   933.4 3460.35   954.8 3462.12     970  3471.2  1055.2 3503.04  1094.2 3522.61
  1141.9 3534.85  1159.2 3542.63  1193.9 3550.28  1216.3 3557.32    1407 3577.09
#Mann= 7 ,-1,0
       0      .1       0     310     .06       0     410      .1       0
   701.2    .045       0   847.8    .025       0     910     .12       0
 1123.01      .1       0
Bank Sta=701.2,847.8
XS Rating Curve= 0 ,0
Exp/Cntr(USF)=0,0
Exp/Cntr=0.3,0.1

Type RM Length L Ch R = 1 ,263835  ,543.2,581.8,617.5
XS GIS Cut Line= 4
2299270.96845856611983.7710742732299872.02620231612174.835787519
2300556.67475811612023.5762228662300799.01024785612087.600980783
#Sta/Elev= 30
       0 3670.91   106.2  3643.3   116.6 3643.57   139.8 3633.86   240.5 3603.37
     362 3584.38   493.2  3548.2   513.3  3539.5   530.1  3527.6   563.7 3524.58
   584.2 3511.68   613.6 3499.81   622.5 3493.85   634.9 3479.79   671.8 3456.83
   684.1 3451.73   692.6 3443.48   699.3 3440.49   819.3 3440.44   835.7 3446.59
   870.4 3445.92   888.9 3451.35   913.5 3453.71  1015.9 3448.31  1077.4  3450.8
  1134.7 3461.54  1301.8  3474.7  1401.5 3491.89    1480 3513.28  1582.5 3536.23
#Mann= 7 ,-1,0
       0      .1       0     450     .06       0     610      .1       0
   699.3    .045       0   819.3      .1       0  820.69     .12       0
  920.69      .1       0
Bank Sta=699.3,819.3
XS Rating Curve= 0 ,0
Exp/Cntr(USF)=0,0
Exp/Cntr=0.3,0.1

Type RM Length L Ch R = 1 ,263253  ,562.8,569.4,584.8
XS GIS Cut Line= 2
2299163.49455736612230.5629955492300321.82438141612915.211551346
#Sta/Elev= 30
       0  3612.1    98.8 3583.79   189.3 3553.47   230.2 3544.76   293.5 3527.55
   343.2 3511.59   355.8 3504.73   370.4 3503.91     498  3473.8   553.7 3466.41
     579 3460.54   598.2  3452.3   659.5 3449.07     788 3452.94   814.3 3447.74
   823.2 3442.96   852.2 3439.65   854.1 3439.61   934.7 3439.66   966.1 3451.52
    1007 3454.31  1018.7 3462.43    1037 3469.85  1176.5 3500.62  1196.8 3508.04
  1208.9 3509.48  1252.3 3521.29  1269.8 3528.46  1320.4 3536.24  1345.5 3546.99
#Mann= 5 ,-1,0
       0      .1       0     370     .06       0     460      .1       0
   852.2    .045       0   934.7      .1       0
Bank Sta=852.2,934.7
XS Rating Curve= 0 ,0
Exp/Cntr(USF)=0,0
Exp/Cntr=0.3,0.1

Type RM Length L Ch R = 1 ,262683  ,404.3,383.7,369
XS GIS Cut Line= 2
2298940.58572524612365.9005007652299657.07839991613217.730680651
#Sta/Elev= 30
       0 3622.02      56 3597.88     144 3570.37   186.6 3553.19   229.3 3531.68
   334.2 3501.92   380.6 3482.63   396.3 3482.39   421.9 3472.02   464.2 3463.19
   507.4 3457.97     574 3455.92   589.7 3452.03   605.4 3452.43   615.8  3456.6
   632.3 3453.38   720.2 3449.45   737.3 3444.98   748.7 3438.55   751.5 3438.29
   861.5 3438.48   884.9 3451.06   903.3  3451.4   908.5 3454.97   929.4 3477.38
   945.1 3484.01  1021.2 3506.47    1062 3514.14  1080.6 3520.81  1113.1 3528.03
#Mann= 6 ,-1,0
       0      .1       0     350     .06       0     500      .1       0
   748.7    .045       0   861.5      .1       0     970     .12       0
Bank Sta=748.7,861.5
XS Rating Curve= 0 ,0
Exp/Cntr(USF)=0,0
Exp/Cntr=0.3,0.1

Type RM Length L Ch R = 1 ,262300  ,291.9,269.7,253.2
XS GIS Cut Line= 4
2298557.78325842612681.0750496562298650.00814051612970.938759376
2299274.94897342613265.4968589632299497.85780554613257.535829244
#Sta/Elev= 30
       0 3550.22    67.3 3526.44    97.5 3519.36   172.2 3496.09   205.8 3493.78
   239.4 3484.74   306.6 3476.64   346.6  3476.5   487.8 3466.63   525.2 3467.53
   547.9 3461.87     572  3460.9     590 3464.06   642.7  3457.4   712.9 3453.46
   746.3 3442.97   770.3 3442.04   778.5 3446.25     793 3446.01   819.5 3437.44
     908 3437.44   938.6 3445.17   948.1 3449.93   974.7 3451.01  1000.4 3463.53
  1040.3 3476.84  1092.3 3490.35  1136.4 3496.72  1184.4  3510.3  1218.1 3510.59
#Mann= 11 ,-1,0
       0      .1       0     140     .06       0     240      .1       0
  334.18     .06       0  384.18      .1       0  764.18     .06       0
   819.5    .045       0     908    .025       0  984.18      .1       0
 1085.06     .12       0 1185.06      .1       0
Bank Sta=819.5,908
XS Rating Curve= 0 ,0
Exp/Cntr(USF)=0,0
Exp/Cntr=0.3,0.1

Type RM Length L Ch R = 1 ,262030  ,1008.5,913.1,818.2
XS GIS Cut Line= 4
2298469.87541134613582.7482560272298681.85225939613460.542087067
2299338.63721117613480.444661364 2299521.7408947613269.477373822
#Sta/Elev= 30
       0 3568.59   104.2 3533.35   201.2 3495.36   233.5 3487.47   244.7 3482.35
     275 3473.32     291 3465.85     315 3458.72   347.1 3455.07   403.1 3454.98
   443.1 3448.47   495.1  3449.4   507.1 3451.82   579.2 3449.35   591.2 3443.92
   603.2 3441.28   611.2 3436.89   715.2 3436.69   716.9 3436.92   751.2 3450.04
   771.2  3451.6   783.3 3449.98   803.3 3458.71   891.3 3461.02   944.9 3466.54
   961.9 3471.94  1038.5 3486.81  1111.6 3496.46    1166 3510.84  1181.1 3512.73
#Mann= 7 ,-1,0
       0      .1       0  434.68     .06       0  534.68      .1       0
   611.2    .045       0   716.9      .1       0  824.68     .12       0
 1141.77      .1       0
#XS Ineff= 2 , 0
           510.3 3482.98
Permanent Ineff=
       F       F
Bank Sta=611.2,716.9
XS Rating Curve= 0 ,0
Exp/Cntr(USF)=0,0
Exp/Cntr=0.3,0.1

Type RM Length L Ch R = 1 ,261117  ,637.6,633.6,630
XS GIS Cut Line= 3
2299796.39641999614256.6450589242299712.80560794613524.230324816
2299731.38077643613245.345183257
#Sta/Elev= 30
       0 3561.27    15.6 3556.46    27.6 3549.11    51.8 3547.48      80 3538.28
   112.2 3524.98   116.2 3521.78   124.3 3510.78   136.3 3503.26   164.5 3498.72
   200.8 3485.17   216.9 3482.77     241  3473.5   265.2 3461.26   293.4 3453.05
   305.4 3446.47   317.5 3443.12   333.6 3433.75   454.4 3433.75   466.5 3438.81
   490.6 3442.51   510.8  3449.5   527.3 3448.52   627.5 3452.65   760.3 3463.18
   776.3 3466.93   804.4 3469.99   840.4 3481.03   948.7 3501.28  1016.7 3519.16
#Mann= 6 ,-1,0
       0     .06       0      80      .1       0   333.6    .045       0
   454.4    .025       0     470      .1       0     570     .12       0
Bank Sta=333.6,454.4
XS Rating Curve= 0 ,0
Exp/Cntr(USF)=0,0
Exp/Cntr=0.3,0.1

Type RM Length L Ch R = 1 ,260483  ,649.6,668.6,697.3
XS GIS Cut Line= 4
2300369.59055972614324.3138115322300425.31776775614021.794682226
2300325.80489627 613500.347235662300352.09199307613224.862507381
#Sta/Elev= 30
       0 3556.82    23.5 3552.08    76.4 3534.11    92.7 3515.92   117.1 3506.21
   133.3 3502.24   153.7  3493.7   197.2  3482.8   214.7  3480.2   247.2 3470.42
   259.4 3469.55     292 3460.71   340.8 3453.57     410 3448.55   511.8 3444.34
     520 3442.32   540.4 3430.83     691  3430.8   695.1 3432.44   699.2 3437.47
   711.4  3439.9   731.7  3447.6   756.2 3447.61     918 3477.73   986.3 3505.77
  1034.5 3521.45  1070.7 3536.93  1086.8 3540.43  1106.8 3552.44  1115.2 3554.53
#Mann= 6 ,-1,0
       0     .06       0      50      .1       0  347.61     .12       0
   540.4    .045       0     691      .1       0  848.47     .12       0
Bank Sta=540.4,691
XS Rating Curve= 0 ,0
Exp/Cntr(USF)=0,0
Exp/Cntr=0.3,0.1

Type RM Length L Ch R = 1 ,259815  ,1038.7,1094.1,1148.1
XS GIS Cut Line= 2
2300895.01852115614384.0215344212301124.39547709613282.000722541
#Sta/Elev= 30
       0 3540.06    68.3 3512.89     105 3506.29   154.1 3480.92   190.8 3468.91
   276.6 3451.03   358.4 3442.72   464.6 3442.97   517.7    3440   525.9 3442.56
   558.6 3440.44   599.4 3441.38     628 3436.98   636.2 3430.28   640.3 3429.34
   734.2 3429.34   746.5 3434.26   758.8 3443.48     771 3446.91   783.3 3445.95
   790.9 3447.89   821.8 3467.43   836.4 3478.99   897.7 3497.91   975.3  3535.5
  1012.1 3549.69  1073.4 3580.37  1097.9    3589  1110.1 3597.01  1125.6 3598.87
#Mann= 8 ,-1,0
       0     .12       0     110      .1       0     200     .12       0
     610    .025       0   640.3    .045       0   734.2     .12       0
     810      .1       0    1010     .06       0
Bank Sta=640.3,734.2
XS Rating Curve= 0 ,0
Exp/Cntr(USF)=0,0
Exp/Cntr=0.3,0.1

Type RM Length L Ch R = 1 ,258721  ,765.1,794.2,830.1
XS GIS Cut Line= 3
2300914.92109545614475.5733761852301949.85495886614284.508662939
2302260.33511788614395.963078999
#Sta/Elev= 30
       0 3557.67      42 3555.65    78.6 3547.67   115.2 3545.03   130.2 3539.84
   159.9  3537.5   274.4 3513.53   371.4 3500.88   416.2 3476.56   463.2    3445
   475.9 3438.77   492.4 3434.77   574.8 3433.48   595.1 3435.13   611.4 3433.25
   781.8 3435.94   831.1 3434.02   875.8 3427.32   969.4  3427.5   977.5  3429.3
   989.7  3439.6   993.8 3440.94  1022.2 3442.11  1071.9 3470.76  1101.7 3473.38
  1186.1 3488.55  1216.4 3497.04  1241.9 3501.03  1314.3 3523.28  1382.3 3539.48
#Mann= 5 ,-1,0
       0     .12       0     730      .1       0   875.8    .045       0
   969.4    .025       0    1030      .1       0
Bank Sta=875.8,969.4
XS Rating Curve= 0 ,0
Exp/Cntr(USF)=0,0
Exp/Cntr=0.3,0.1

Type RM Length L Ch R = 1 ,257926  ,534.1,549.7,573
XS GIS Cut Line= 2
2300879.09646171 614666.638089432301826.45899822615164.202446841
#Sta/Elev= 30
       0  3544.3    11.6 3543.89    23.8 3531.13    46.4 3526.17      60 3519.49
   100.6 3507.64   124.1 3498.39   168.4 3489.34   198.2  3486.3   218.1 3482.18
   275.2 3459.69   334.5 3443.29   430.4 3438.58     435 3436.02   448.5 3422.59
   452.8  3421.7     453 3421.66   532.9 3421.76   556.9 3425.79     599 3429.27
   657.3 3431.89   715.1 3431.86   733.2  3436.2   755.7 3431.75   791.9 3440.43
   823.5 3458.05   867.7 3478.19   906.2 3492.93   986.2 3512.25  1070.1 3529.42
#Mann= 6 ,-1,0
       0     .12       0      30      .1       0     240     .12       0
   452.8    .045       0   532.9    .025       0     620      .1       0
#XS Ineff= 2 , 0
                          741.53         3456.49
Permanent Ineff=
       F       F
Bank Sta=452.8,532.9
XS Rating Curve= 0 ,0
Exp/Cntr(USF)=0,0
Exp/Cntr=0.3,0.1

Type RM Length L Ch R = 1 ,257377  ,635.9,632.5,647
XS GIS Cut Line= 2
2300763.66153079614726.3458123192301197.53765046 615665.74731911
#Sta/Elev= 30
       0 3541.03    25.2 3531.97    29.6 3528.09    38.7 3514.02    47.2 3509.61
    87.1 3504.67   141.2 3489.14   183.8 3480.18     219 3462.04   258.7 3455.34
   279.8 3447.87     325 3438.47   346.8 3438.25   404.1 3431.74   472.7 3432.47
   496.6 3426.16   597.9 3431.19     620 3425.82   637.6 3418.54   664.93418.378
   725.9 3418.35   747.7 3429.78   791.8 3432.95   801.2 3441.46   840.3 3459.51
   871.1 3479.18   897.7 3479.27   915.2 3487.03   985.7 3505.43  1034.8 3527.31
#Mann= 10 ,-1,0
       0      .1       0     180     .12       0     280      .1       0
     410     .12       0     490      .1       0     600    .025       0
   664.9    .045       0   725.9      .1       0     820     .06       0
     930      .1       0
#XS Ineff= 2 , 0
          526.79 3440.83
Permanent Ineff=
       F       F
Bank Sta=664.9,725.9
XS Rating Curve= 0 ,0
Exp/Cntr(USF)=0,0
Exp/Cntr=0.3,0.1

Type RM Length L Ch R = 1 ,256744  ,746.9,712.3,671.8
BEGIN DESCRIPTION:
Structure XS 4
END DESCRIPTION:
XS GIS Cut Line= 2
2300454.95509804614683.545366082 2300450.0300599615697.591437984
#Sta/Elev= 30
       0 3553.41    37.6 3541.19    77.6 3540.51   101.6 3529.99   121.6 3515.87
   181.6 3491.97   257.6 3467.22   277.6 3464.85   300.3 3459.01   313.6 3452.75
   345.6  3443.5   405.6 3434.47   453.6    3425     490 3422.02   509.3 3419.83
   517.4 3415.26   517.6 3415.16   661.6 3415.34   694.2 3423.05   706.3 3427.92
   769.6 3429.12   789.6 3432.56   817.6 3441.33   853.6 3440.24   865.6 3444.63
   900.1 3450.52   925.6 3458.17   975.7    3475  1001.6 3489.27  1014.1 3492.09
#Mann= 7 ,-1,0
       0     .06       0     100      .1       0     490    .025       0
   517.4    .045       0   661.6      .1       0     690     .07       0
     790      .1       0
Bank Sta=517.4,661.6
XS Rating Curve= 0 ,0
Exp/Cntr(USF)=0,0
Exp/Cntr=0.3,0.1

Type RM Length L Ch R = 1 ,256032  ,62.2,62,62.1
BEGIN DESCRIPTION:
Structure XS 3
END DESCRIPTION:
XS GIS Cut Line= 3
2299202.96870579615149.7732932962299649.11737019615247.793258885
2300385.51261916615765.260190592
#Sta/Elev= 30
       0 3646.63    38.1 3624.92      79 3610.66     120 3579.97   181.8 3546.68
   197.8 3541.03   214.2  3539.5   263.3 3523.41   296.1 3503.91     333 3485.96
   348.8 3482.49   390.3    3454     419  3439.3   447.6 3430.66   507.9 3422.39
   520.3 3422.69   534.6 3427.16   563.2 3426.49   597.4  3410.8   602.3 3410.62
   670.7 3410.64   738.5 3423.73   959.2 3423.25  1022.7 3443.16  1106.2 3449.69
    1141 3457.11  1223.2 3463.57  1266.8 3472.76  1311.2 3489.83  1356.8 3492.26
#Mann= 8 ,-1,0
       0      .1       0  466.79     .06       0  586.79     .07       0
   597.4    .045       0   670.7     .08       0  706.79     .07       0
  826.79     .08       0  836.79      .1       0
#XS Ineff= 2 , 0
          537.76 3453.88
Permanent Ineff=
       F       F
Bank Sta=597.4,670.7
XS Rating Curve= 0 ,0
Exp/Cntr(USF)=0,0
Exp/Cntr=0.3,0.1

Type RM Length L Ch R = 1 ,255970  ,386.7,372.6,348.9
BEGIN DESCRIPTION:
Structure XS 2
END DESCRIPTION:
XS GIS Cut Line= 3
2299182.48602991615240.4959320712299641.15634048615319.442526352
2300369.59055972615820.987398622
#Sta/Elev= 30
       0  3654.9    17.9 3638.26    50.4 3614.24    78.8 3597.91    95.1 3593.02
   147.8 3559.54   180.3 3544.53   204.7 3541.81   241.2 3530.08   269.6  3510.5
   322.4 3487.49   338.6 3475.79   350.8 3474.43   371.1 3458.92   389.9 3449.87
   455.7 3427.18   483.2 3423.46   529.2 3423.91   571.1  3410.7   575.9 3410.59
   653.6 3410.59   692.5 3425.27   917.5 3422.92   993.6 3448.47  1035.4 3457.13
  1100.4 3460.36  1221.8 3460.24  1286.7 3471.75  1323.8 3484.95  1349.8 3485.42
#Mann= 6 ,-1,0
       0      .1       0  485.41     .06       0  555.41      .1       0
   571.1    .045       0   653.6     .08       0  725.41      .1       0
Bank Sta=571.1,653.6
XS Rating Curve= 0 ,0
Exp/Cntr(USF)=0,0
Exp/Cntr=0.3,0.1

Type RM Length L Ch R = 1 ,255597  ,642.2,595.9,557.3
BEGIN DESCRIPTION:
Structure XS 1
END DESCRIPTION:
XS GIS Cut Line= 3
2299143.67558439615672.4645443452299955.61701436615797.104309467
2300325.80489627615836.909458059
#Sta/Elev= 30
       0  3578.5    16.7 3573.95      41 3559.98    81.8 3545.91    89.5 3541.53
   101.7 3530.66   134.1 3530.09   158.3  3514.7   182.6 3506.04   197.5 3502.85
   336.4 3452.68   401.1 3435.99   461.8 3424.95   486.1 3415.84   494.2 3409.56
   498.3 3409.19   595.4 3409.12   597.3 3409.27     652 3415.06   684.4 3421.01
   785.6 3423.61   793.9 3422.28   797.7 3422.92   813.9 3434.28     826 3438.95
   846.2 3445.34   910.5 3459.39   982.9 3461.56  1143.9 3460.94  1193.8 3472.55
#Mann= 3 ,-1,0
       0      .1       0   498.3    .045       0   597.3      .1       0
Bank Sta=498.3,597.3
XS Rating Curve= 0 ,0
Exp/Cntr(USF)=0,0
Exp/Cntr=0.3,0.1

Type RM Length L Ch R = 1 ,255001  ,872.5,832.4,803.1
XS GIS Cut Line= 2
2299525.72140956616617.0903704792300325.80489627615860.792547215
#Sta/Elev= 30
       0 3647.75    35.6 3627.04    52.3  3611.3    63.9 3593.78    69.7 3589.99
   116.3 3570.21   162.9 3543.77   197.8 3529.53   209.5 3520.66     228  3519.6
     262 3505.27   310.1 3477.34   321.4 3469.08   337.6 3449.68   349.2 3428.26
     361 3414.75   377.7 3404.98   465.7 3404.59   468.5 3404.89   505.3 3408.48
   533.6 3416.21   593.8 3413.62   663.7 3418.78   779.8 3418.81   803.4 3424.26
   844.2 3445.06   867.5 3453.01   937.4 3458.95  1038.2 3460.64    1101 3471.49
#Mann= 3 ,-1,0
       0      .1       0   377.7    .045       0   468.5      .1       0
Bank Sta=377.7,468.5
XS Rating Curve= 0 ,0
Exp/Cntr(USF)=0,0
Exp/Cntr=0.3,0.1

Type RM Length L Ch R = 1 ,254169  ,633.6,667.5,698.4
XS GIS Cut Line= 3
2300496.96703522616911.6484700662300648.22659987616577.285221886
2300672.10968903615896.617180949
#Sta/Elev= 30
       0 3583.61    29.1 3572.11    82.9 3545.43   108.1 3526.02   134.4 3526.44
   156.4 3513.67   191.5 3501.28   209.8 3490.92   226.6 3484.71   248.6 3471.72
   279.4 3465.03   336.8 3440.67   371.1 3423.02   395.1  3415.7   431.1 3410.32
   467.2 3408.27   483.2 3404.68   491.2 3400.15   615.2 3400.09     616 3400.13
   631.3 3407.93   683.3 3414.87   739.3 3411.91   787.4 3412.29   800.1 3417.48
   899.4 3443.75   955.5 3453.72  1019.5 3475.09  1031.5 3476.95  1048.1 3487.46
#Mann= 3 ,-1,0
       0      .1       0   491.2    .045       0     616      .1       0
#XS Ineff= 2 , 0
                           725.2          3426.9
Permanent Ineff=
       F       F
Bank Sta=491.2,616
XS Rating Curve= 0 ,0
Exp/Cntr(USF)=0,0
Exp/Cntr=0.3,0.1

Type RM Length L Ch R = 1 ,253501  ,615.2,624.1,629.4
XS GIS Cut Line= 2
2300795.50564967617043.0054604222301661.68138178616135.780775239
#Sta/Elev= 30
       0 3558.37    10.3 3555.49    30.2 3539.58    49.9 3539.04    68.9 3532.63
     214 3500.25   234.8 3479.84   259.2 3477.02   281.9 3469.45   361.1 3434.44
   429.6 3411.61   468.6 3407.53     644 3408.25     661 3406.36   689.3 3396.74
   692.1 3396.69   771.3 3396.69   779.8 3400.04   788.7 3407.96   815.5 3410.93
   826.5 3409.27   850.5 3427.88   910.4 3440.12   942.7  3449.5  1089.9 3501.66
  1130.6 3521.46  1169.4 3547.71  1187.2  3551.1    1207 3565.91  1254.3 3583.53
#Mann= 3 ,-1,0
       0      .1       0   689.3    .045       0   771.3      .1       0
#XS Ineff= 2 , 0
          526.64 3429.31
Permanent Ineff=
       F       F
Bank Sta=689.3,771.3
XS Rating Curve= 0 ,0
Exp/Cntr(USF)=0,0
Exp/Cntr=0.3,0.1

Type RM Length L Ch R = 1 ,252877  ,416.3,406.5,395.9
XS GIS Cut Line= 4
2300979.02563726617198.7437427532301316.95309623 617222.12862909
2301826.45899822616875.8238363322302132.95864239 616609.12934076
#Sta/Elev= 30
       0 3512.21   185.6 3499.53   189.6 3496.59   201.6 3473.85   205.6    3469
   217.7 3464.94   237.7 3450.01   269.8  3432.1   313.9 3422.84   497.2 3401.85
   528.9 3400.55   553.9 3404.67   603.7 3402.85   637.7 3398.13   647.3 3394.31
     755 3394.39   787.6  3399.6   805.3 3407.29   850.5 3405.67   860.1 3410.17
   909.7 3417.13   999.5 3423.69  1025.9 3432.91  1063.1 3436.95  1096.8 3450.13
  1163.9 3466.58  1283.9 3501.22  1322.9 3518.34  1342.7 3520.58  1361.1 3532.28
#Mann= 5 ,-1,0
       0      .1       0  488.74     .06       0   647.3    .045       0
     755     .12       0  828.74      .1       0
Bank Sta=647.3,755
XS Rating Curve= 0 ,0
Exp/Cntr(USF)=0,0
Exp/Cntr=0.3,0.1

Type RM Length L Ch R = 1 ,252471  ,369.7,362.3,354.7
XS GIS Cut Line= 3
2301488.11523518618018.2316009462301607.53068096 617556.49187727
2302351.88695965616875.823836332
#Sta/Elev= 30
       0 3536.11    71.3 3525.46   170.5 3504.74   385.3 3430.34   537.4 3413.64
   604.3 3409.84     630 3405.41   647.8 3398.57   683.8 3392.56   695.2 3392.47
   819.3 3392.59   833.6 3400.87   862.6 3403.52   884.6 3399.69   910.1 3403.63
   932.7 3401.31   975.2 3400.79     995 3404.22  1056.8 3405.41  1082.8 3409.03
    1122 3416.75  1181.3 3436.06    1281 3457.59  1296.3  3459.1  1317.9 3466.46
  1366.7 3474.48  1394.7 3481.57  1445.2 3498.77  1473.5 3500.63  1485.6 3506.28
#Mann= 6 ,-1,0
       0      .1       0  636.93    .025       0  666.93      .1       0
   683.8    .045       0   819.3    .025       0  906.93      .1       0
#XS Ineff= 2 , 0
                          910.32         3415.86
Permanent Ineff=
       F       F
Bank Sta=683.8,819.3
XS Rating Curve= 0 ,0
Exp/Cntr(USF)=0,0
Exp/Cntr=0.3,0.1

Type RM Length L Ch R = 1 ,252109  ,516.6,506.5,496.2
XS GIS Cut Line= 3
2301822.47848336618237.1599182072301933.93289942617779.400709389
2302582.75682149617023.102886126
#Sta/Elev= 30
       0 3618.03    79.3 3614.49   119.4 3602.55   127.2 3597.23   152.3 3571.43
   197.6 3551.98     247 3522.68   292.3 3504.38   337.6 3468.69   362.3 3456.91
   399.3 3433.38   432.3 3423.72   448.7 3424.09   480.7 3417.97   574.2 3409.58
   590.6 3403.41   611.1 3390.65   616.4 3390.37   729.6 3390.74   753.4 3398.21
   812.5 3398.45   837.7 3401.74   854.4 3397.23   890.4 3398.14  1058.2 3417.79
  1268.6 3467.08    1331  3483.8    1348 3484.86  1365.3 3492.91  1467.6 3514.43
#Mann= 8 ,-1,0
       0      .1       0     320     .12       0     410      .1       0
     430     .12       0  541.13      .1       0   611.1    .045       0
   729.6    .025       0  751.13      .1       0
#XS Ineff= 2 , 0
                          837.55         3419.31
Permanent Ineff=
       F       F
Bank Sta=611.1,729.6
XS Rating Curve= 0 ,0
Exp/Cntr(USF)=0,0
Exp/Cntr=0.3,0.1

Type RM Length L Ch R = 1 ,251602  ,591.9,579.7,566.1
XS GIS Cut Line= 2
2302192.66636528618396.3805125782302897.21749537 617218.14811423
#Sta/Elev= 30
       0 3558.74    30.2 3541.24    73.6 3520.17   240.7 3466.18     288 3449.15
     342 3423.87   413.9 3397.09   433.6 3393.64     489 3395.25   507.1 3388.22
   632.9 3388.27   656.2 3394.04     699 3395.02   716.1  3400.1   744.8 3398.55
   754.1 3400.33     796 3399.72     810 3403.11   856.6 3403.66   934.3 3409.66
   991.8 3425.04  1061.7 3449.43  1098.6  3458.4  1129.2 3462.59  1140.9 3470.11
  1187.5 3487.76  1280.7 3513.38  1300.6 3520.53  1336.7 3528.42  1372.8 3540.39
#Mann= 7 ,-1,0
       0      .1       0     440    .025       0   507.1    .045       0
   632.9    .025       0     670      .1       0     900     .12       0
    1000      .1       0
#XS Ineff= 2 , 0
                          714.66         3415.69
Permanent Ineff=
       F       F
Bank Sta=507.1,632.9
XS Rating Curve= 0 ,0
Exp/Cntr(USF)=0,0
Exp/Cntr=0.3,0.1

Type RM Length L Ch R = 1 ,251022  ,506.5,496.8,486.2
XS GIS Cut Line= 2
2302849.45131706618643.1724338542303227.60022869 617389.31025318
#Sta/Elev= 30
       0 3556.57    64.8 3531.66   106.5 3507.85   181.7  3472.6     236 3454.96
   365.6 3403.92   398.6 3388.45   415.7 3385.53   520.1 3385.54   561.9 3398.27
   729.2  3394.7   751.7 3397.43   766.6 3403.56   783.4 3397.92   804.2 3398.16
   825.1 3407.55   958.8 3416.62  1000.6 3436.36  1018.1 3440.11  1034.6  3452.2
    1063 3465.16  1092.5  3474.5  1109.2 3482.62  1138.5 3490.33  1163.6 3503.47
  1201.2 3515.77  1238.8 3538.11  1263.8 3549.52    1291 3567.28  1309.6 3575.04
#Mann= 7 ,-1,0
       0      .1       0     340    .025       0   415.7    .045       0
   520.1    .025       0     550      .1       0     750     .12       0
    1270      .1       0
Bank Sta=415.7,520.1
XS Rating Curve= 0 ,0
Exp/Cntr(USF)=0,0
Exp/Cntr=0.3,0.1

Type RM Length L Ch R = 1 ,250526  ,734.4,746.9,785.1
XS GIS Cut Line= 2
2303428.78258045618758.6073647732303543.38660582617525.227859975
#Sta/Elev= 30
       0 3568.81    21.5 3568.34    26.5 3561.47    45.6 3516.36    69.7 3500.61
   105.9 3495.13   154.1 3476.35   222.4  3456.5   290.1  3426.9   326.8 3418.81
   386.7 3400.13   431.3 3394.94   443.3 3391.58   459.4 3383.05     588 3383.01
     604  3390.4   620.1 3394.11   692.4 3393.53   744.6 3396.95   756.7 3394.75
     825 3404.72   885.2 3419.13     905 3420.82   913.3 3425.17   953.5 3435.76
   967.5 3436.75  1009.8 3447.07    1074 3478.69  1162.6  3497.6  1238.7 3518.99
#Mann= 5 ,-1,0
       0      .1       0   459.4    .045       0     588    .025       0
     640      .1       0    1140     .12       0
#XS Ineff= 2 , 0
                          749.03         3419.83
Permanent Ineff=
       F       F
Bank Sta=459.4,588
XS Rating Curve= 0 ,0
Exp/Cntr(USF)=0,0
Exp/Cntr=0.3,0.1

Type RM Length L Ch R = 1 ,249779  ,700.8,719.1,771
XS GIS Cut Line= 4
2303565.94399173 618774.529424212303921.86822018 618597.06466152
2304333.35415658618281.609284563 2304769.4687838618165.925252234
#Sta/Elev= 30
       0 3524.38    20.6 3520.81    60.6 3506.41   100.8 3502.97   136.6  3495.1
   190.2 3489.84   244.3 3492.17   275.1 3480.17   330.7 3463.92   334.7  3460.5
   342.7 3445.21   346.7 3440.55   357.6 3434.14   391.4 3421.66   430.4 3398.72
     446 3392.12   476.3 3387.87   531.7 3391.63   602.2 3392.11   708.1 3378.86
   713.1 3378.78   763.5 3378.84   795.8 3393.67   811.7 3392.59   864.3 3408.44
   884.5 3409.83   910.3 3418.24  1179.8 3464.33  1316.4 3496.95  1367.4 3512.03
#Mann= 6 ,-1,0
       0      .1       0  537.71    .025       0  607.71      .1       0
   708.1    .045       0   763.5      .1       0  857.71     .12       0
#XS Ineff= 2 , 0
          533.72 3407.79
Permanent Ineff=
       F       F
Bank Sta=708.1,763.5
XS Rating Curve= 0 ,0
Exp/Cntr(USF)=0,0
Exp/Cntr=0.3,0.1

Type RM Length L Ch R = 1 ,249060  ,337.6,347.7,377
XS GIS Cut Line= 2
2303506.23626884618850.1592065362304664.56609289619319.859959932
#Sta/Elev= 30
       0 3515.94      28  3508.1    40.9 3502.56      99 3488.98   118.6 3481.42
   175.8 3471.17   226.5  3457.5   295.6 3442.31   312.9 3436.51   464.5 3407.01
     486 3400.19   495.2 3394.65   507.5 3390.83   538.2 3376.78   541.2 3376.53
   684.1 3376.88   697.9    3383   719.4 3388.93   735.9 3387.34   796.1 3399.86
   817.9 3401.36   904.2 3413.59   912.8 3416.34   934.4 3418.67   964.6 3426.68
   999.2 3431.55  1055.3 3444.53  1137.9  3474.2  1163.2 3480.46  1249.9 3511.51
#Mann= 3 ,-1,0
       0      .1       0   538.2    .045       0   684.1      .1       0
Bank Sta=538.2,684.1
XS Rating Curve= 0 ,0
Exp/Cntr(USF)=0,0
Exp/Cntr=0.3,0.1

Type RM Length L Ch R = 1 ,248712  ,409.9,415.2,421.1
XS GIS Cut Line= 4
2303283.32743672619013.3603157672303601.76862546619192.483484435
2304083.41092344619498.983128599 2304409.8131419619686.067326986
#Sta/Elev= 30
       0 3548.63    26.9 3531.27    73.1 3506.36    88.6 3494.41   111.1 3482.72
   147.8 3472.77   175.4 3470.95   203.2 3464.85   253.4 3448.41   303.9 3440.34
   326.8 3432.38   364.7 3427.92   418.8 3414.48   489.3 3402.51   553.5 3397.33
   567.3 3391.49     582 3374.93   586.3 3373.31   666.9 3373.45   692.1    3377
   755.9 3377.28   818.6 3386.87     837 3385.39   895.6 3392.24   940.7 3401.26
  1013.1 3423.78  1158.4 3476.12  1190.5  3483.3  1228.6 3502.84  1312.5  3530.4
#Mann= 6 ,-1,0
       0      .1       0  475.36     .12       0   586.3    .045       0
   666.9      .1       0  705.36    .025       0  765.36      .1       0
Bank Sta=586.3,666.9
XS Rating Curve= 0 ,0
Exp/Cntr(USF)=0,0
Exp/Cntr=0.3,0.1

Type RM Length L Ch R = 1 ,248297  ,477.1,503.5,554.8
XS GIS Cut Line= 3
2303072.36014918 619104.912157532303315.17155559619447.236435429
2303995.83959653620024.411090025
#Sta/Elev= 30
       0 3564.78    19.9  3555.7      46 3547.73    83.3 3529.78      89  3524.8
    98.4 3508.27   132.7 3488.31   177.9 3467.98   255.3 3440.48   377.9 3411.21
   412.3 3400.66   457.7 3396.92   509.8 3396.55   641.3 3386.75   651.7 3384.86
   671.5 3373.26   682.9 3370.67   788.1 3370.53   830.9 3377.93   843.3 3382.41
     872 3385.42   886.6 3384.05   972.4 3407.39  1053.6 3438.05  1094.4 3448.96
  1115.4 3457.62  1135.9 3470.33  1186.7 3487.35  1239.1 3512.48  1312.1 3541.02
#Mann= 8 ,-1,0
       0      .1       0     390     .12       0  509.69      .1       0
  529.69     .12       0  659.69    .025       0   682.9    .045       0
   788.1    .025       0  789.69      .1       0
Bank Sta=682.9,788.1
XS Rating Curve= 0 ,0
Exp/Cntr(USF)=0,0
Exp/Cntr=0.3,0.1

Type RM Length L Ch R = 1 ,247793  ,460.1,457.7,455
XS GIS Cut Line= 4
2302809.64616846 619164.619880422303056.43808974619570.632396067
2303124.10684235620036.3526346032303323.13258531620346.832793627
#Sta/Elev= 30
       0 3604.69      28 3588.55    37.2 3576.73    42.8 3572.93      99 3547.86
   173.9 3506.67     230 3469.69   300.2 3434.64   359.1 3419.29     436 3407.25
   451.5 3402.72   635.3 3380.28   655.6 3381.39   675.8 3377.88   691.9 3378.57
   708.1 3374.38   720.2 3368.06   833.4    3368   853.6 3378.76   869.8 3382.12
   885.9 3381.57   902.1 3393.74   914.2 3398.48   965.7 3412.49  1027.5 3433.07
  1065.5 3442.32  1179.5 3478.96  1224.3 3490.67  1303.1 3507.08  1314.5 3511.36
#Mann= 4 ,-1,0
       0      .1       0  705.13    .025       0   720.2    .045       0
   833.4      .1       0
Bank Sta=720.2,833.4
XS Rating Curve= 0 ,0
Exp/Cntr(USF)=0,0
Exp/Cntr=0.3,0.1

Type RM Length L Ch R = 1 ,247336  ,568.4,550.8,530.2
XS GIS Cut Line= 4
2302335.96490021 619387.528712542302606.63991064619733.833505297
 2302698.1917524620191.5927141152302909.15903995620510.033902857
#Sta/Elev= 30
       0 3583.35    13.3 3577.58    42.7 3557.84    66.9 3545.67   103.6 3522.25
   186.5 3479.67   243.5 3456.63   291.5 3441.12   318.6 3429.92   377.1 3412.19
   451.1 3400.58   471.5 3393.89   576.3 3380.16     602  3367.8   613.7 3365.56
   687.7 3365.46   699.9 3365.56   728.5 3370.58   744.8 3375.88   785.6 3378.52
   797.8 3376.11   830.5 3381.15   922.7 3409.67   990.3 3422.27  1064.8 3440.35
  1116.7 3449.61  1183.1 3466.54  1229.7 3474.32  1250.4 3480.56  1288.3 3495.88
#Mann= 3 ,-1,0
       0      .1       0   613.7    .045       0   699.9      .1       0
#XS Ineff= 2 , 0
                          788.45            3400
Permanent Ineff=
       F       F
Bank Sta=613.7,699.9
XS Rating Curve= 0 ,0
Exp/Cntr(USF)=0,0
Exp/Cntr=0.3,0.1

Type RM Length L Ch R = 1 ,246785  ,635.4,622.3,606
XS GIS Cut Line= 3
2301794.61487935619805.482772764 2302053.3483452620044.313664321
2302562.85424719620748.864794414
#Sta/Elev= 30
       0 3599.62    34.9 3581.68    40.8 3576.52    51.1 3571.31    56.6 3566.38
    72.9 3539.34    83.8 3528.29    94.3 3520.57   141.1 3491.48     199 3460.35
   312.3 3420.92   370.6 3395.46   403.5 3386.21     455 3377.35   486.6 3362.87
   581.1  3362.9   621.2 3375.49   654.3 3377.16   692.8 3375.74   704.2 3378.13
   759.7 3380.13   802.4 3386.32   821.7 3391.44   850.3 3403.22   889.4 3415.56
  1012.2 3436.77  1116.8  3459.1  1138.1 3467.54  1192.4 3483.56  1221.6  3496.4
#Mann= 4 ,-1,0
       0      .1       0   486.6    .045       0   581.1    .025       0
  632.11      .1       0
Bank Sta=486.6,581.1
XS Rating Curve= 0 ,0
Exp/Cntr(USF)=0,0
Exp/Cntr=0.3,0.1

Type RM Length L Ch R = 1 ,246163  ,677.7,666.5,653.9
XS GIS Cut Line= 2
2301253.26485849620231.3978627082302272.27666246621059.344953438
#Sta/Elev= 30
       0 3562.44    60.4 3550.47   122.8 3530.54   142.9 3519.96   174.1 3512.67
   213.8 3496.66   230.5 3487.84   259.3 3478.33   275.6 3467.88   288.3 3462.72
   313.6 3448.31   398.6 3419.63   426.4 3412.01   436.7 3405.19   465.9 3380.09
     481 3362.22   484.9 3360.27   599.1 3360.24   620.4 3365.79   657.3 3371.52
   735.6 3372.36   771.7 3375.08   838.7 3372.75   890.9 3378.83   947.4 3400.46
  1086.1 3429.53  1140.7  3442.9  1209.8 3469.77  1261.3 3483.17    1313 3502.32
#Mann= 3 ,-1,0
       0      .1       0   484.9    .045       0   599.1      .1       0
#XS Ineff= 2 , 0
                          775.31         3389.22
Permanent Ineff=
       F       F
Bank Sta=484.9,599.1
XS Rating Curve= 0 ,0
Exp/Cntr(USF)=0,0
Exp/Cntr=0.3,0.1

Type RM Length L Ch R = 1 ,245496  ,383.8,390.6,399.2
XS GIS Cut Line= 4
 2300938.8041846620800.6114875852301257.24537334621103.130616891
2301598.07674535621284.8249958492301837.48773849621475.475107599
#Sta/Elev= 30
       0 3477.03    93.7 3454.62   189.5 3435.89   217.1 3428.69   250.2 3417.15
   314.4 3403.16   432.2 3381.08   463.6 3376.55   496.9 3374.27   519.6 3368.51
   528.6 3363.65   548.2 3358.11   637.5 3358.07   673.7 3365.07   691.9 3363.49
   732.6 3368.12   768.9 3368.93   782.5  3370.9   791.8 3369.55   815.5 3374.59
   904.8 3408.18   955.3 3438.37   980.9 3451.34  1003.7 3459.75  1022.5 3464.19
  1042.9 3473.48  1058.2 3482.93  1108.6 3508.65  1119.6  3518.7  1131.5 3523.39
#Mann= 6 ,-1,0
       0      .1       0     120     .12       0     130      .1       0
   548.2    .045       0   637.5    .025       0  639.23      .1       0
Bank Sta=548.2,637.5
XS Rating Curve= 0 ,0
Exp/Cntr(USF)=0,0
Exp/Cntr=0.3,0.1

Type RM Length L Ch R = 1 ,245105  ,392.5,425.9,450.7
XS GIS Cut Line= 2
2300585.11846371621062.6617653942301543.84244321 621771.85711325
#Sta/Elev= 30
       0 3480.72   138.1 3436.96   181.3 3426.39   221.3 3413.97   249.9 3407.92
   293.5 3402.45     362 3385.75   395.8 3380.11   407.8 3375.48   448.2 3375.23
   501.3 3372.38     571 3372.39   593.1 3365.95   655.6 3364.52   675.5 3357.04
   804.6    3357   807.6 3357.02   819.8 3361.01     845 3362.65   869.5 3367.79
   905.5 3367.47   919.2  3369.5   934.2 3368.68   959.1  3380.5  1033.3 3429.64
  1060.2 3443.19  1083.5 3452.36  1127.9 3479.76  1163.1 3496.04  1192.5 3512.75
#Mann= 6 ,-1,0
       0      .1       0      70     .12       0     360      .1       0
   675.5    .045       0   807.6    .025       0     850      .1       0
Bank Sta=675.5,807.6
XS Rating Curve= 0 ,0
Exp/Cntr(USF)=0,0
Exp/Cntr=0.3,0.1

Type RM Length L Ch R = 1 ,244680  ,497.3,491.6,490
XS GIS Cut Line= 4
2300397.45416374621170.7993694982300715.89535248621481.279528522
2300930.84315488621927.0971927622301070.16117496622078.356757415
#Sta/Elev= 30
       0 3486.53    49.2 3467.04    98.8  3451.4   216.1 3425.16   266.4 3412.38
   300.6 3401.82   316.6 3399.41   345.9 3392.19   381.6 3388.92   449.1 3376.69
   466.8 3375.07   507.8 3374.08   540.8 3371.06   644.5 3369.64   693.3 3357.35
   706.6 3355.25   804.6 3355.16   808.8 3355.26     831 3357.15   848.7 3362.74
   862.1 3364.57   884.3 3364.84   897.6 3367.88   912.3 3366.75   950.6 3389.68
  1018.4 3427.32  1040.4 3441.95  1075.1 3460.59  1109.1 3473.69  1145.3 3495.61
#Mann= 3 ,-1,0
       0      .1       0   706.6    .045       0   808.8      .1       0
Bank Sta=706.6,808.8
XS Rating Curve= 0 ,0
Exp/Cntr(USF)=0,0
Exp/Cntr=0.3,0.1

Type RM Length L Ch R = 1 ,244188  ,596.5,579.4,543.7
XS GIS Cut Line= 4
2299895.90929147621588.7534297232300313.86335169621819.623291562
 2300508.9085798622150.0060248822300767.64204565622313.207134113
#Sta/Elev= 30
       0  3579.5    15.2 3571.48    32.9 3565.15    59.4 3550.58    91.9  3535.7
   105.4 3524.67   194.8  3469.8   291.9 3423.74   333.9 3410.97   356.7 3406.27
     407 3390.22   494.9 3377.82   524.1 3368.48     549 3362.98   581.5 3362.08
   597.1 3364.93   651.2 3365.02   683.7 3353.48   799.8 3353.47   812.5 3356.98
   827.7 3365.82   851.2 3368.15   861.1 3377.77   869.7 3383.69   891.9  3390.7
   959.6 3405.13  1082.5 3449.27  1134.6 3463.02    1152 3465.61    1167 3470.86
#Mann= 7 ,-1,0
       0     .12       0      70      .1       0     170     .12       0
     180      .1       0  647.48    .025       0   683.7    .045       0
   799.8      .1       0
#XS Ineff= 2 , 0
          599.57 3384.05
Permanent Ineff=
       F       F
Bank Sta=683.7,799.8
XS Rating Curve= 0 ,0
Exp/Cntr(USF)=0,0
Exp/Cntr=0.3,0.1

Type RM Length L Ch R = 1 ,243608  ,771.9,767.5,752.1
XS GIS Cut Line= 2
 2299501.8383204622173.8891140382300652.20711473 622659.51192687
#Sta/Elev= 30
       0 3562.21   141.7    3507   234.7 3460.69   384.6 3401.43     415 3387.32
   449.7 3366.04   467.1 3357.26   480.6 3357.43   492.8 3350.59   497.5  3349.7
   575.7 3349.72   602.7 3352.52   625.6 3360.79   636.4 3362.18   669.8 3360.04
   688.5 3362.71   701.6 3360.56   727.9 3361.06     771 3365.12   784.1 3363.18
   844.8 3382.61   889.7 3391.99   905.6 3397.89   944.4 3402.39  1035.1 3422.43
  1092.3 3443.31  1166.1 3463.51    1195 3475.09  1210.2 3483.04  1248.7 3496.35
#Mann= 5 ,-1,0
       0      .1       0   497.5    .045       0   575.7      .1       0
     600    .025       0     700      .1       0
Bank Sta=497.5,575.7
XS Rating Curve= 0 ,0
Exp/Cntr(USF)=0,0
Exp/Cntr=0.3,0.1

Type RM Length L Ch R = 1 ,242841  ,586.9,557.3,522.1
XS GIS Cut Line= 3
2299334.07659473623024.1427867082299784.56338545623124.062300609
2300532.79166896623145.134739703
#Sta/Elev= 30
       0 3554.69    26.7 3551.38    67.7 3539.78     133 3516.51   146.8 3514.08
   190.6 3499.19   243.9 3475.06   256.2 3471.25   280.4 3457.38   321.7 3437.42
   395.5  3404.6   436.5 3391.14     469  3376.9   505.1 3364.42   537.1 3360.85
   557.1  3356.2   621.1 3354.61  649.36  3346.5   801.2 3346.25   821.2 3356.21
   837.2 3359.46   849.2 3358.11   853.2 3360.58   861.2 3370.35   881.2 3379.67
   909.2 3388.57   944.7  3395.7  1102.2  3451.5    1151 3463.62    1210  3481.5
#Mann= 6 ,-1,0
       0     .12       0     100      .1       0  531.43     .06       0
  631.43      .1       0  649.36    .045       0   801.2      .1       0
Bank Sta=649.36,801.2
XS Rating Curve= 0 ,0
Exp/Cntr(USF)=0,0
Exp/Cntr=0.3,0.1

Type RM Length L Ch R = 1 ,242284  ,451.7,417.4,370.6
XS GIS Cut Line= 4
2299438.15008265623913.374107544 2299844.1625983623837.744325218
2300317.84386655 623602.893948522300562.14817886623320.028292102
#Sta/Elev= 30
       0 3567.89     6.1 3562.33    38.7 3544.86   107.8 3512.93   173.4  3489.3
   228.3  3459.7     242 3455.56   375.8 3395.96   396.7 3383.52   408.9  3383.1
   439.8 3370.11   506.8 3359.62   546.9    3359   582.7 3351.22   631.8    3351
   666.4 3347.44   680.9 3349.39   721.1 3346.84   738.9 3342.31   765.5 3342.28
   850.5 3342.39     855 3343.32   868.4 3353.65   941.7 3358.79   961.6 3371.16
     981  3376.6  1117.6 3397.18  1218.8 3429.88  1261.1  3437.6  1315.5 3458.33
#Mann= 5 ,-1,0
       0      .1       0     330     .06       0     423      .1       0
   738.9    .045       0   850.5      .1       0
Bank Sta=738.9,850.5
XS Rating Curve= 0 ,0
Exp/Cntr(USF)=0,0
Exp/Cntr=0.3,0.1

Type RM Length L Ch R = 1 ,241866  ,567.1,543,507.4
XS GIS Cut Line= 4
2300382.02860456624525.0459900672300325.80489627624176.088088257
2300469.10343121623686.4847605652300628.32402558623356.102027245
#Sta/Elev= 30
       0 3545.79   129.5 3497.46   182.9  3460.4   230.8 3429.55   255.1 3418.72
   271.3 3414.59   295.6 3400.93   344.3 3381.85   381.5 3360.11   389.8 3352.99
   448.2 3340.31   554.4 3340.54   594.1  3342.6   615.6 3348.69   635.7 3351.62
   685.7 3348.55   702.4 3351.03   723.3 3349.51   760.7 3351.59   773.3 3355.56
   834.9  3357.4   844.6  3356.2   852.5 3360.27   860.8 3367.42   869.5 3370.45
   918.3 3380.03    1056 3401.83  1104.8  3415.9  1140.3 3423.24  1230.3 3451.66
#Mann= 7 ,-1,0
       0      .1       0     310     .12       0  413.46    .025       0
  423.46      .1       0   448.2    .045       0   554.4    .025       0
  613.46      .1       0
#XS Ineff= 2 , 0
                          647.94          3369.4
Permanent Ineff=
       F       F
Bank Sta=448.2,554.4
XS Rating Curve= 0 ,0
Exp/Cntr(USF)=0,0
Exp/Cntr=0.3,0.1

Type RM Length L Ch R = 1 ,241323  ,727.6,691.5,629.4
XS GIS Cut Line= 4
2300883.07697657624482.5877324222300926.86264002624088.516761353
2300819.38873882623718.3288794392300763.66153079623344.160482667
#Sta/Elev= 30
       0 3535.78      24 3535.45    37.6 3532.86    81.9 3513.16   110.1 3504.46
   134.2 3500.15   158.4 3487.24   186.5 3464.24   208.7 3449.98   299.2 3403.97
   307.3 3402.11     400 3364.92   420.8 3360.93   441.6 3352.53   474.9 3348.43
   491.6 3338.61   508.3    3336     566 3335.94   604.1 3336.05   645.7 3345.14
     679 3342.97     704  3344.4   733.2 3354.31   753.2 3351.65   770.7 3353.22
   791.2  3364.3   803.4 3367.11  1037.9 3411.46  1102.5 3429.74  1160.3 3452.02
#Mann= 4 ,-1,0
       0      .1       0   466.5    .025       0   508.3    .045       0
   604.1      .1       0
Bank Sta=508.3,604.1
XS Rating Curve= 0 ,0
Exp/Cntr(USF)=0,0
Exp/Cntr=0.3,0.1

Type RM Length L Ch R = 1 ,240632  ,581.4,594.5,615.5
XS GIS Cut Line= 4
 2301858.3031171623885.5105035292301583.64759181623622.796522817
2301209.47919503623431.7318095712300998.51190749623172.998343718
#Sta/Elev= 30
       0 3522.07    58.3 3503.66      81 3493.06   145.2 3457.53     169 3438.64
   191.4 3424.79   270.5 3392.36   307.2 3378.76   365.1 3363.86   401.9 3351.97
   418.8 3351.05   471.6 3335.82   490.9 3333.96   496.3 3333.85     631    3334
   642.5 3336.41   662.4  3350.2   698.4 3355.08   725.3 3355.99   738.8 3349.66
   761.2 3350.64   774.7 3360.75   783.7 3361.94   865.5 3388.66     948 3407.68
   962.1 3413.05  1040.9  3431.9  1118.5 3469.01  1128.6 3471.71    1134 3475.62
#Mann= 4 ,-1,0
       0      .1       0  450.07    .025       0   490.9    .045       0
     631      .1       0
Bank Sta=490.9,631
XS Rating Curve= 0 ,0
Exp/Cntr(USF)=0,0
Exp/Cntr=0.3,0.1

Type RM Length L Ch R = 1 ,240037  ,534.2,534.1,534.4
XS GIS Cut Line= 2
2302113.05606809623415.8097501342301444.32957173622719.219649759
#Sta/Elev= 30
       0 3459.54    36.4 3445.71    73.2 3435.35    97.9 3430.56   135.4 3419.13
     231  3379.9   388.3 3346.03   417.1 3331.73   469.3 3329.35     550 3329.11
   552.6 3329.23     557 3330.57   562.6  3335.3   573.9 3341.42   584.6 3344.81
   599.4 3343.83   615.1 3349.95   702.3  3363.3   721.1 3367.11   746.4 3375.63
   780.5 3391.28   813.2 3409.57   825.7 3418.24   835.4 3420.58   850.3 3432.76
   867.7 3441.25   908.1 3465.87   924.7 3477.69     937 3483.03   965.6 3504.19
#Mann= 4 ,-1,0
       0      .1       0   469.3    .045       0   552.6    .025       0
     570      .1       0
Bank Sta=469.3,552.6
XS Rating Curve= 0 ,0
Exp/Cntr(USF)=0,0
Exp/Cntr=0.3,0.1

Type RM Length L Ch R = 1 ,239503  ,555.1,565.8,577
XS GIS Cut Line= 2
 2302523.0490986623081.4465019542301866.26414682 622380.87588672
#Sta/Elev= 30
       0 3482.34    38.7 3464.22    67.3 3455.69     132 3429.72   181.3 3398.21
   226.4 3389.32   252.6 3379.61   285.5 3372.03   334.8 3357.94   356.8 3353.41
   367.3 3353.39   426.7  3345.1     437  3341.8   460.4 3329.43   477.6 3325.28
   520.1 3325.26     589  3325.3   593.7 3326.54   606.6  3336.1   612.4 3338.33
   641.9 3341.44   653.1  3341.1   678.6 3355.56   740.6 3374.31   795.4 3395.42
   828.6 3410.79   855.7 3425.11   881.5 3434.26   919.1 3452.09   960.3 3478.84
#Mann= 3 ,-1,0
       0      .1       0   477.6    .045       0     589      .1       0
Bank Sta=477.6,589
XS Rating Curve= 0 ,0
Exp/Cntr(USF)=0,0
Exp/Cntr=0.3,0.1

Type RM Length L Ch R = 1 ,238937  ,564.7,573.2,586.5
XS GIS Cut Line= 2
2302944.98367368622898.3428184272302351.88695965621927.097192762
#Sta/Elev= 30
       0    3478    71.7 3453.22   139.7 3434.59   170.1 3423.17   216.5 3408.83
   296.6 3390.79   400.7 3360.07   418.5 3356.51   474.7 3350.29   498.2 3344.78
   508.1 3344.17   526.3 3335.76   573.2 3322.74   577.8 3322.69   669.3 3322.73
   684.6 3327.93   692.3 3333.79   696.9 3335.53   732.5 3339.31   746.6 3337.97
   760.6 3345.51   848.2 3363.85   868.8 3370.78   901.2 3377.98   945.6 3391.22
   996.6 3408.94  1045.4 3430.57  1068.4 3443.62  1098.1 3456.64    1138  3481.4
#Mann= 3 ,-1,0
       0      .1       0   573.2    .045       0   669.3      .1       0
Bank Sta=573.2,669.3
XS Rating Curve= 0 ,0
Exp/Cntr(USF)=0,0
Exp/Cntr=0.3,0.1

Type RM Length L Ch R = 1 ,238364  ,525.1,536.5,553.1
XS GIS Cut Line= 2
2303315.17155559622703.2975903222302980.80830741621632.539093175
#Sta/Elev= 30
       0 3514.11    39.9 3498.88    69.3 3484.84   157.3  3457.5   169.3 3451.32
   190.8  3436.1   215.9 3425.66   245.3 3419.21   291.4  3400.5   312.3 3396.41
   320.7 3392.42   345.8 3386.14   412.8 3354.93   429.6  3348.9   551.2 3334.68
   593.1  3319.3   681.1 3319.31   697.8 3323.94   714.6 3333.66   739.7 3336.81
   748.1 3335.78   798.4  3350.9   823.6 3355.32   890.6 3373.89     899 3378.83
   911.6    3379   940.9 3392.65  1020.5  3423.7  1083.3 3451.38  1121.7 3471.06
#Mann= 5 ,-1,0
       0      .1       0     580     .05       0   593.1    .045       0
   681.1     .05       0     730      .1       0
Bank Sta=593.1,681.1
XS Rating Curve= 0 ,0
Exp/Cntr(USF)=0,0
Exp/Cntr=0.3,0.1
