HEC-RAS study SHAVERSFK.prj: SHAVERSFK

--- SHAVERSFK.g01 (geometry) --- (continued)

Type RM Length L Ch R = 1 ,237828  ,413.5,422.4,436
XS GIS Cut Line= 2
2303645.55428891622667.4729565892303669.43737807621576.811885145
#Sta/Elev= 30
       0 3534.66    18.3 3530.07    70.3 3506.15   126.5  3485.4   222.3 3436.83
   254.4 3429.87   274.4  3422.7   286.4  3421.2   329.8 3406.77   342.4 3401.48
   394.4 3373.31   466.4 3344.25   494.4 3336.34   551.9 3330.01   566.4 3324.23
   590.4 3317.47   674.5 3317.47   686.5 3320.84   706.5 3330.15   742.5 3335.36
   758.5 3335.73   766.5 3341.42   838.5 3362.88   914.5  3393.2   926.5 3394.72
   956.9 3409.99   970.5 3418.46  1006.5 3434.42  1022.5 3443.12  1090.9 3469.27
#Mann= 4 ,-1,0
       0      .1       0   590.4    .045       0   674.5    .025       0
     710      .1       0
Bank Sta=590.4,674.5
XS Rating Curve= 0 ,0
Exp/Cntr(USF)=0,0
Exp/Cntr=0.3,0.1

Type RM Length L Ch R = 1 ,237405  ,509.7,515.8,524.7
XS GIS Cut Line= 2
 2303832.6384873622707.2781051812304270.49512182621588.753429723
#Sta/Elev= 30
       0 3548.11   140.2  3503.7   169.8 3491.25   195.7 3475.15   207.2 3469.91
   251.4 3453.43   322.2 3432.51   371.7  3412.6   393.2 3400.94   427.5 3378.77
   444.7 3370.28   496.2  3336.1   541.5 3326.89   577.9  3323.4   599.3 3318.41
   646.6 3315.59     668 3315.44   706.7 3315.47   723.9 3322.75   732.9  3329.5
   745.4 3332.51   758.3 3331.95   779.2 3344.22   814.1 3356.82   934.4 3390.48
  1024.6 3432.68  1037.5 3435.47  1044.7  3440.1  1081.7 3454.26  1201.2 3494.38
#Mann= 3 ,-1,0
       0      .1       0   646.6    .045       0   706.7      .1       0
Bank Sta=646.6,706.7
XS Rating Curve= 0 ,0
Exp/Cntr(USF)=0,0
Exp/Cntr=0.3,0.1

Type RM Length L Ch R = 1 ,236889  ,649.9,675.4,711.9
XS GIS Cut Line= 3
2304206.80688407622834.6545806792304636.70248888  622157.9670546
2304760.09844951621819.623291561
#Sta/Elev= 30
       0 3506.93   101.3 3463.74   120.9  3459.7   143.9  3452.4   158.1 3451.05
   167.2 3446.76   218.9 3433.76   252.9 3422.21   352.4 3377.71   399.1 3360.53
   448.3 3336.02   494.7 3322.63     523 3322.11   535.3 3319.96   546.7 3316.04
   569.5 3313.29   669.9  3313.2   674.7 3313.85   698.4 3326.31   717.3 3330.32
   731.5 3329.65     741 3336.72   770.9 3345.35   811.1 3364.75   845.1 3383.17
   866.4  3390.4   985.6 3443.89  1100.6 3483.34  1130.4 3492.13  1161.8 3499.33
#Mann= 3 ,-1,0
       0      .1       0   569.5    .045       0   669.9      .1       0
Bank Sta=569.5,669.9
XS Rating Curve= 0 ,0
Exp/Cntr(USF)=0,0
Exp/Cntr=0.3,0.1

Type RM Length L Ch R = 1 ,236214  ,395.7,406.4,426.8
XS GIS Cut Line= 3
2304278.45615154 622993.875175052305098.44221255622766.985828071
2305389.01979728622774.946857789
#Sta/Elev= 30
       0 3503.41    10.1 3499.36      64 3466.46   142.9 3439.31   213.3 3411.59
     230  3402.7   317.2 3376.98   362.8  3360.4   450.6 3341.96   495.7 3328.23
     533 3322.69   574.5 3323.61   607.7 3313.93   657.5 3308.08   732.2 3308.21
   748.8 3311.14   761.3 3315.59   769.6 3321.38   811.1 3325.26   837.4 3348.56
   864.5 3379.05   884.5 3392.02   909.1 3405.44   948.6 3419.44   992.6 3438.38
  1016.6 3452.36  1032.6    3467  1060.6 3481.17  1108.6 3497.27  1141.5 3512.05
#Mann= 6 ,-1,0
       0      .1       0     520     .12       0     550      .1       0
   657.5    .045       0   732.2      .1       0  1120.8     .12       0
Bank Sta=657.5,732.2
XS Rating Curve= 0 ,0
Exp/Cntr(USF)=0,0
Exp/Cntr=0.3,0.1

Type RM Length L Ch R = 1 ,235808  ,470.7,470.5,461.5
XS GIS Cut Line= 2
 2304282.4366664623129.2126802662305321.35104467 623268.53070034
#Sta/Elev= 30
       0 3508.89      30 3489.94    74.4 3466.15   108.3 3456.98   151.1 3442.34
   183.8 3426.84   219.7 3407.24     252 3394.35   292.3 3382.46   377.1  3350.4
   486.1 3322.06   530.4 3308.26   578.9 3307.06   586.9 3305.08     595 3305.04
   691.9 3305.28   691.9 3305.29   712.1 3310.63   728.2 3321.47   744.3 3321.74
   760.5  3335.7   773.7 3349.55   795.1 3360.19     813 3371.36   861.4 3393.16
   881.6 3405.05   921.9 3422.14   950.2 3439.12  1006.7 3466.01  1048.2 3480.46
#Mann= 4 ,-1,0
       0      .1       0     300     .12       0   586.9    .045       0
   691.9      .1       0
Bank Sta=586.9,691.9
XS Rating Curve= 0 ,0
Exp/Cntr(USF)=0,0
Exp/Cntr=0.3,0.1

Type RM Length L Ch R = 1 ,235337  ,499.8,493.5,482.7
XS GIS Cut Line= 2
2304167.00173548623670.562701128 2305289.5069258623634.738067394
#Sta/Elev= 30
       0 3523.23    17.2 3513.32    41.2 3494.71    77.2 3475.28    93.2 3464.02
   156.9 3433.97   221.3 3406.94   241.3 3395.67   329.3 3362.79   377.4 3346.78
   413.4 3337.72   437.4 3334.63   517.4 3317.65  558.283301.792   569.5 3299.32
   621.5 3299.47   641.5 3301.71   669.5 3305.43   677.5 3311.41   689.5 3315.01
   713.5 3317.52   729.5 3317.15   741.6 3323.97   789.4 3337.21   837.6 3357.31
   877.6  3377.2     901 3385.33   925.6 3398.85   969.7 3418.72  1123.1 3474.06
#Mann= 4 ,-1,0
       0      .1       0  558.28    .045       0   641.5      .1       0
     810     .12       0
Bank Sta=558.28,641.5
XS Rating Curve= 0 ,0
Exp/Cntr(USF)=0,0
Exp/Cntr=0.3,0.1

Type RM Length L Ch R = 1 ,234844  ,570.1,558,546
XS GIS Cut Line= 2
2304326.22232985624311.4255934732305365.13670813623941.237711559
#Sta/Elev= 30
       0 3485.17   113.9 3431.51   184.7 3404.09   227.1 3383.78   252.6 3375.86
   295.1 3355.48   354.5 3336.16   413.4 3320.97   443.7 3317.82   466.6 3312.56
   479.2 3305.22   507.3 3295.85   507.4 3295.84   554.1 3295.84   609.3 3302.19
   620.1 3305.29   630.5 3311.02   643.3 3314.07   657.6 3314.16   668.7  3322.5
   715.5 3345.14     724 3346.39   770.3 3362.23   817.4 3372.73   944.8 3426.98
   961.7 3431.67    1002 3447.85  1033.9 3456.03  1080.6 3474.79  1102.9  3481.1
#Mann= 4 ,-1,0
       0      .1       0   507.3    .045       0   554.1      .1       0
     900     .12       0
Bank Sta=507.3,554.1
XS Rating Curve= 0 ,0
Exp/Cntr(USF)=0,0
Exp/Cntr=0.3,0.1

Type RM Length L Ch R = 1 ,234286  ,653.1,639.2,625.9
XS GIS Cut Line= 2
 2304712.3322712624920.4443669432305588.04554024624235.795811146
#Sta/Elev= 30
       0 3491.91    39.3 3471.09    50.6 3463.09    65.8 3456.57    89.7  3441.2
   121.7 3433.77   193.1 3406.77   226.1 3390.35   238.4 3381.74     304 3347.52
     317 3343.64   361.3 3321.28   407.9 3308.84   429.6 3294.73   436.5 3293.14
   543.1 3293.21   588.8 3305.08   626.3 3309.26   639.6 3308.73   649.7 3316.94
   654.7 3319.11   680.4 3323.14   700.4 3328.78   831.4 3384.13   848.5 3389.34
   874.2 3401.19     934 3423.69  1040.7 3467.55  1071.1    3477  1111.6 3496.94
#Mann= 10 ,-1,0
       0      .1       0      80     .12       0     170      .1       0
   436.5    .045       0   543.1    .025       0     580     .12       0
     650      .1       0     710     .12       0     810      .1       0
     830     .12       0
Bank Sta=436.5,543.1
XS Rating Curve= 0 ,0
Exp/Cntr(USF)=0,0
Exp/Cntr=0.3,0.1

Type RM Length L Ch R = 1 ,233646  ,745.5,724.2,700.7
XS GIS Cut Line= 3
2305006.89037079625398.1061500572305412.90288644625226.944011108
2305970.17496674624550.256485029
#Sta/Elev= 30
       0 3510.75   102.5 3489.69     136  3475.5   153.3 3470.62     175 3461.29
   201.1 3445.07   227.1 3432.14   257.5 3423.17   325.4 3391.68   377.3 3358.01
   453.3 3320.08   489.8 3308.84   515.2  3305.9   540.1 3290.45   541.4 3290.31
   672.3 3290.41   686.4 3296.27   711.3 3300.82   779.3 3302.82   795.3 3314.45
   807.9 3320.13   857.4 3332.79   997.4 3385.42  1012.5 3393.12  1069.4 3410.46
  1160.3 3447.41  1199.4 3466.99  1231.3 3479.81  1297.9 3500.48  1317.2 3513.48
#Mann= 8 ,-1,0
       0      .1       0  470.62    .025       0   540.1    .045       0
   672.3      .1       0  680.62     .12       0  830.62      .1       0
  980.62     .12       0 1300.62      .1       0
Bank Sta=540.1,672.3
XS Rating Curve= 0 ,0
Exp/Cntr(USF)=0,0
Exp/Cntr=0.3,0.1

Type RM Length L Ch R = 1 ,232922  ,622.3,594.2,561.5
XS GIS Cut Line= 4
2306117.45401653625943.4366857792306077.64886794625636.937041614
2306201.04482857625226.9440111082306252.79152175624852.775614335
#Sta/Elev= 30
       0 3463.39    58.7 3448.81      95 3437.54   147.5 3412.93   159.6 3409.21
   187.8 3391.21   227.3 3369.28   304.8 3336.44   354.8 3311.42   392.4 3299.12
   409.1 3290.95   442.5 3285.53   542.1 3285.53   584.5 3290.38   601.2 3297.75
   634.6 3300.81   647.2 3299.26   659.7  3302.7   709.8  3307.3   787.5 3339.11
   880.3 3373.53   904.3 3385.85   932.8 3396.82   957.1 3403.08   997.5 3419.19
  1013.6 3422.49  1037.8 3435.91    1054    3451  1078.2 3456.01    1115  3468.9
#Mann= 5 ,-1,0
       0      .1       0  349.07    .025       0   442.5    .045       0
   542.1    .025       0  559.07      .1       0
Bank Sta=442.5,542.1
XS Rating Curve= 0 ,0
Exp/Cntr(USF)=0,0
Exp/Cntr=0.3,0.1

Type RM Length L Ch R = 1 ,232328  ,576.5,546,510.8
XS GIS Cut Line= 2
2306845.88823578625863.8263885932306495.60292816 624880.63921835
#Sta/Elev= 30
       0 3507.15    32.5  3490.3     172 3385.54   191.3 3369.05   206.6 3353.91
   232.1 3333.83     257 3320.56   297.7 3289.11   325.5 3282.65   342.5 3283.88
   355.3 3280.92   413.6 3280.82   448.7 3281.02     473  3283.8   491.1 3292.68
   529.3 3298.41   576.1 3297.25   588.6  3298.6   597.3 3296.43     627  3296.5
   682.2 3305.58     711 3315.77   732.1 3327.14   762.9 3338.81   788.4 3347.24
   822.3 3355.35   881.8 3378.91   924.3 3389.61   979.5 3407.36  1043.7 3423.66
#Mann= 3 ,-1,0
       0      .1       0   355.3    .045       0   448.7      .1       0
Bank Sta=355.3,448.7
XS Rating Curve= 0 ,0
Exp/Cntr(USF)=0,0
Exp/Cntr=0.3,0.1

Type RM Length L Ch R = 1 ,231782  ,481.3,497.6,511.1
XS GIS Cut Line= 4
2307331.51104861625342.3789420272307180.25148396625151.314228781
2306969.28419642625039.8598127212306698.60918598624701.516049682
#Sta/Elev= 30
       0  3451.4    16.8 3440.94    31.2 3435.13    98.5 3398.25   134.2 3375.31
   169.9 3357.37   215.8 3323.34   252.8  3301.9   280.8 3290.43   301.6 3284.73
   310.4 3280.02   325.2 3275.62   325.2 3275.61   334.1 3275.59   402.4 3275.61
   420.2 3281.17   433.8 3292.71   484.1 3295.93   496.4 3304.74   567.5 3328.27
   661.4 3353.69   681.3 3360.79   690.6 3360.44     721  3368.8   762.3 3383.57
   843.6 3404.66   869.9 3414.41   880.2 3416.16   894.8 3423.23   915.6 3429.74
#Mann= 5 ,-1,0
       0      .1       0   325.2    .045       0   402.4      .1       0
  652.29     .12       0  852.29      .1       0
Bank Sta=325.2,402.4
XS Rating Curve= 0 ,0
Exp/Cntr(USF)=0,0
Exp/Cntr=0.3,0.1

Type RM Length L Ch R = 1 ,231284  ,436.3,439,441.3
XS GIS Cut Line= 4
2307641.99120764625067.7234167362307438.98494981624836.853554898
 2307283.7448703624590.0616336222307017.05037473624311.425593473
#Sta/Elev= 30
       0 3452.65    51.3    3423     130 3383.27     159 3366.52   285.7 3306.04
     307 3298.64   330.7 3293.19   354.3 3283.61   377.9 3279.71   392.1 3275.12
   440.4 3275.73   468.8 3271.51   519.7 3271.36   523.9 3271.51   538.6 3277.96
   552.9 3288.79   570.3 3292.14   584.8 3290.78   590.6 3292.11   611.3 3307.92
   655.9 3332.65   666.7 3335.96   683.3 3347.07   699.9 3353.01   757.7 3384.89
   771.9 3387.67     794 3398.04   888.1 3424.04   922.3 3436.82   984.7 3465.39
#Mann= 7 ,-1,0
       0      .1       0  327.43     .12       0  337.43      .1       0
   468.8    .045       0   523.9      .1       0  678.99     .12       0
  698.99      .1       0
Bank Sta=468.8,523.9
XS Rating Curve= 0 ,0
Exp/Cntr(USF)=0,0
Exp/Cntr=0.3,0.1

Type RM Length L Ch R = 1 ,230845  ,432.8,459.5,479.4
XS GIS Cut Line= 2
 2307928.5882775624868.6976737722307486.75112812624008.906464167
#Sta/Elev= 30
       0  3462.7    26.7 3456.67    53.4 3446.35    83.1 3425.67   107.4  3411.1
   152.4 3388.34   197.3 3361.58   219.8 3350.65   273.8 3332.33   324.7 3307.53
   354.7 3296.82   377.2 3292.25     401 3280.26   412.9 3277.62   426.7 3270.35
   440.2 3266.97   498.7 3267.02   513.9 3272.07   530.1 3283.99   543.6 3286.22
   557.1 3285.25   575.1 3296.47   620.1 3311.34     683 3336.44     755 3361.29
   777.5 3372.59   858.5 3405.45   889.9 3420.96   934.9 3438.16   966.7 3452.54
#Mann= 4 ,-1,0
       0      .1       0   440.2    .045       0   498.7      .1       0
     880     .12       0
Bank Sta=440.2,498.7
XS Rating Curve= 0 ,0
Exp/Cntr(USF)=0,0
Exp/Cntr=0.3,0.1

Type RM Length L Ch R = 1 ,230386  ,496.8,519.2,532.1
XS GIS Cut Line= 2
2308024.12063413624884.6197332092308247.02946625623965.120800715
#Sta/Elev= 30
       0 3473.88    26.1 3469.17    42.6 3463.19    61.2 3447.45   122.2 3419.98
   143.5 3402.59   164.1 3390.92   246.4 3354.61   283.4 3328.07   328.7 3303.22
   369.9 3293.49   406.9 3278.08   423.4 3276.46   448.1 3268.52   493.2 3265.48
   493.3 3265.47   563.3 3265.63   583.9 3269.61   592.1 3278.91   599.2 3282.93
   616.8 3282.33     624 3284.84   641.5 3298.55     658 3307.49   715.6 3346.37
     732 3361.03   785.6 3389.93   849.1 3417.79   904.9 3436.57   946.1 3458.11
#Mann= 5 ,-1,0
       0      .1       0     480    .025       0   493.2    .045       0
   563.3    .025       0     680      .1       0
Bank Sta=493.2,563.3
XS Rating Curve= 0 ,0
Exp/Cntr(USF)=0,0
Exp/Cntr=0.3,0.1

Type RM Length L Ch R = 1 ,229867  ,263.8,276.5,289
XS GIS Cut Line= 2
2308254.99049596624996.074149269   2308848.08721624339.289197488
#Sta/Elev= 30
       0 3468.62    65.2 3429.23    82.2  3417.1     102 3399.15   164.3 3362.84
   192.6 3338.04     241 3302.79   270.3 3275.33   284.2 3271.18   294.6 3263.27
   305.7 3257.81   311.1 3257.66   371.8 3257.82   402.7 3265.79     422 3273.72
   470.2 3276.75   484.3 3287.29   497.1 3294.27   518.3 3301.85   532.9 3306.46
   586.3 3317.32   612.9  3320.2   628.4 3327.23   652.3 3334.37     718 3372.62
   736.9 3385.58   759.1 3396.98   790.8 3417.35   855.3 3451.32   884.9  3463.8
#Mann= 3 ,-1,0
       0      .1       0   305.7    .045       0   371.8      .1       0
Bank Sta=305.7,371.8
XS Rating Curve= 0 ,0
Exp/Cntr(USF)=0,0
Exp/Cntr=0.3,0.1

Type RM Length L Ch R = 1 ,229590  ,332.8,336.4,340.1
XS GIS Cut Line= 2
2308358.48388231625107.5285653292309138.66479473624697.535534823
#Sta/Elev= 30
       0 3463.24      48 3422.39    87.8  3395.5   127.4    3374   137.5 3365.67
   146.5 3351.82     151 3347.18   202.8 3307.13   254.4 3278.09     273 3271.65
   282.1 3270.52   304.7 3260.04   313.7 3259.07   322.7 3255.62     394 3255.19
  395.963255.549   426.7 3271.37   438.4 3274.44   453.8 3274.35     468  3284.5
     517  3303.2   555.4 3310.74   584.8 3314.08     630 3327.96   666.5 3337.42
   684.3 3344.45   697.8  3354.4   720.4 3366.69   837.9 3439.33   881.3 3460.67
#Mann= 5 ,-1,0
       0      .1       0   322.7    .045       0  395.96      .1       0
     620     .12       0     630      .1       0
Bank Sta=322.7,395.96
XS Rating Curve= 0 ,0
Exp/Cntr(USF)=0,0
Exp/Cntr=0.3,0.1

Type RM Length L Ch R = 1 ,229254  ,367.9,375,385.3
XS GIS Cut Line= 2
 2308485.8603578625374.2230609012309242.15818107625079.664961314
#Sta/Elev= 30
       0 3451.65    32.5 3431.52    48.9 3407.14      52 3404.57   109.8 3371.18
   139.8 3345.63   208.5  3296.1   234.3 3280.58   247.2  3277.4   268.6 3267.93
   281.5 3266.04   302.3 3254.72   324.4 3251.57   380.2 3251.68   414.6 3268.05
   440.3 3270.97   448.9 3269.46   461.8 3279.95   521.9 3296.87   547.7 3310.26
   586.5 3322.44   609.1 3332.79   617.4    3334   694.6 3372.43   715.1 3384.72
   723.7 3392.66   732.2 3393.98   770.9  3412.4   784.2 3420.88   811.6 3432.12
#Mann= 6 ,-1,0
       0      .1       0   324.4    .045       0   380.2      .1       0
     560     .12       0     730      .1       0     770     .12       0
Bank Sta=324.4,380.2
XS Rating Curve= 0 ,0
Exp/Cntr(USF)=0,0
Exp/Cntr=0.3,0.1

Type RM Length L Ch R = 1 ,228879  ,369.9,379.6,396.8
XS GIS Cut Line= 2
2308545.56808069625636.9370416142309349.63208227625577.229318725
#Sta/Elev= 30
       0 3410.59    26.7 3390.73    46.7 3377.76    58.8 3372.45    86.8 3356.15
     155 3322.21   239.3 3284.66   263.6 3276.37   275.4 3270.96   291.4 3268.67
   307.5 3259.56   315.5  3258.1   335.5 3247.31   339.5 3247.16   395.7 3247.23
   411.7 3252.36   419.8    3259   435.3 3266.71   451.8 3265.88   467.9  3274.5
     512 3286.96   532.1  3290.8   548.1 3296.22   552.1 3299.16   592.2 3311.31
   632.3 3330.59   660.4 3341.53   692.5 3359.62   704.5  3365.1   806.3 3406.84
#Mann= 4 ,-1,0
       0      .1       0   335.5    .045       0   395.7      .1       0
     760     .12       0
Bank Sta=335.5,395.7
XS Rating Curve= 0 ,0
Exp/Cntr(USF)=0,0
Exp/Cntr=0.3,0.1

Type RM Length L Ch R = 1 ,228499  ,362.4,373.7,391.4
XS GIS Cut Line= 2
 2308485.8603578625859.8458737342309250.11921079626106.637795009
#Sta/Elev= 30
       0  3427.2    15.6 3418.01    65.5 3384.32    78.1 3372.51    99.1  3365.6
   123.6 3352.85   153.8 3341.04   171.3 3332.11   208.4 3309.62   250.4 3290.23
   271.4 3278.61     292 3271.18   347.1  3257.5   363.9 3249.36   380.7 3243.95
   456.4  3243.8   473.2 3248.19   485.8 3255.03   506.8  3263.8   515.2  3264.4
   523.7 3262.89   527.9 3264.78   571.6 3294.87   603.7 3314.99   641.3  3342.9
     654 3350.13   670.8  3356.5     696 3369.91   754.8  3395.6   803.1 3410.87
#Mann= 5 ,-1,0
       0      .1       0     140     .12       0     240      .1       0
   380.7    .045       0   456.4      .1       0
Bank Sta=380.7,456.4
XS Rating Curve= 0 ,0
Exp/Cntr(USF)=0,0
Exp/Cntr=0.3,0.1

Type RM Length L Ch R = 1 ,228125  ,408,431.1,444.6
XS GIS Cut Line= 2
2308334.60079315626023.0469829642309035.17140838626580.319063264
#Sta/Elev= 30
       0 3431.22      14 3427.22    73.8 3394.46   114.5 3377.01   150.7 3357.16
   170.7 3342.24   189.8 3332.58   216.1 3323.65   324.3 3278.66   376.1 3267.45
   385.3 3263.57   395.5 3256.11   405.8  3254.2   426.8 3241.95   431.3 3241.12
   517.5 3241.09   517.9  3241.1   552.1 3246.85   584.7 3259.82   606.1 3262.38
   620.5 3261.92   639.5 3277.48     692 3306.05   722.7  3329.6   761.6 3354.83
     784 3364.98   799.4 3369.75   825.9 3384.11   839.6 3388.87   895.2 3419.45
#Mann= 5 ,-1,0
       0      .1       0     230     .12       0     280      .1       0
   431.3    .045       0   517.9      .1       0
Bank Sta=431.3,517.9
XS Rating Curve= 0 ,0
Exp/Cntr(USF)=0,0
Exp/Cntr=0.3,0.1

Type RM Length L Ch R = 1 ,227694  ,386.9,401.5,405.8
XS GIS Cut Line= 2
2308171.39968392626106.6377950092308537.60705097626950.506945177
#Sta/Elev= 30
       0 3415.41    20.2 3407.95    63.3  3397.8   105.9 3381.57   212.3 3329.82
   229.5 3322.84   268.8  3301.4   373.4 3270.11     404 3264.79   421.4 3255.64
   447.5 3245.73     486 3237.75   546.8 3237.69   550.3 3237.72   565.3 3240.36
   578.3 3253.23   600.1 3253.33   630.7 3256.57   635.1 3260.68   644.1 3274.04
   652.5  3280.2   696.1 3300.08   709.2 3302.36   722.2 3307.36   750.6 3328.34
   787.1 3345.75   823.5 3369.51     846 3380.79   883.6 3403.88   919.9 3420.54
#Mann= 3 ,-1,0
       0      .1       0     486    .045       0   550.3      .1       0
Bank Sta=486,550.3
XS Rating Curve= 0 ,0
Exp/Cntr(USF)=0,0
Exp/Cntr=0.3,0.1

Type RM Length L Ch R = 1 ,227293  ,443.3,437.4,431.6
XS GIS Cut Line= 2
2307924.60776264626142.4624287432308040.04269356627042.058786941
#Sta/Elev= 30
       0 3419.51    51.1 3391.07   168.1 3355.02   220.1 3335.99   268.9  3314.1
     309 3290.74   333.4 3268.54   341.6 3263.07   357.6 3246.79   365.7 3241.85
   381.8 3236.65     402  3236.9   418.1 3241.96   446.3 3240.64   474.6 3235.02
   478.6 3234.85   551.2 3234.96   563.3 3238.68   575.4 3245.18   587.5 3246.01
   599.6 3250.35   615.7 3252.82     644 3252.99   676.2 3265.33   720.6 3294.65
     773 3342.56   784.8 3347.68   797.2 3356.45   877.9 3400.93     907 3422.56
#Mann= 5 ,-1,0
       0     .12       0     260      .1       0     450    .025       0
   474.6    .045       0   551.2      .1       0
Bank Sta=474.6,551.2
XS Rating Curve= 0 ,0
Exp/Cntr(USF)=0,0
Exp/Cntr=0.3,0.1

Type RM Length L Ch R = 1 ,226855  ,393.1,381,371.8
XS GIS Cut Line= 3
2307454.90700925626261.8778745212307622.08863334626850.994073695
 2307713.6404751627057.980846378
#Sta/Elev= 30
       0 3421.56    20.1 3410.81   103.2 3360.79     124 3350.01   198.9 3318.69
   223.8 3310.74   269.3 3288.11   273.7 3285.49   298.4 3262.88   315.3 3250.94
   337.3 3230.26   409.3 3229.81   414.9  3229.9   452.5  3234.7     465 3234.16
   485.8 3239.83   499.2 3240.01   514.9 3245.67   568.9 3248.13   585.5 3251.24
     598 3250.34   602.2 3251.65   614.8 3263.77   632.3 3275.36   667.2 3291.57
   715.4 3323.66     781 3354.76   820.3  3378.4   833.5    3391   838.7 3393.54
#Mann= 3 ,-1,0
       0      .1       0   337.3    .045       0   414.9      .1       0
Bank Sta=337.3,414.9
XS Rating Curve= 0 ,0
Exp/Cntr(USF)=0,0
Exp/Cntr=0.3,0.1

Type RM Length L Ch R = 1 ,226474  ,589.8,546.3,487.6
XS GIS Cut Line= 3
2307001.12831529626409.1569243152307331.51104861626998.273123489
2307614.12760362627169.435262438
#Sta/Elev= 30
       0    3431      14 3420.07    45.9 3400.99    59.6 3388.86    73.4 3383.84
   100.9 3366.76   163.9  3333.6   216.7 3300.43   266.7 3279.55   319.6 3249.18
   357.9 3237.56   362.3 3235.05   366.9 3228.95   371.5  3227.9   505.1 3227.84
   513.5 3229.21   522.8 3238.08   529.6 3241.73   600.8 3241.58   635.9 3248.58
   651.6 3248.05   718.3 3282.76   727.7 3283.42   758.3 3295.65   793.1 3304.33
   827.8 3318.46   874.1 3340.93   935.9 3366.23   970.8 3383.03  1005.8 3394.61
#Mann= 3 ,-1,0
       0      .1       0   371.5    .045       0   505.1      .1       0
Bank Sta=371.5,505.1
XS Rating Curve= 0 ,0
Exp/Cntr(USF)=0,0
Exp/Cntr=0.3,0.1

Type RM Length L Ch R = 1 ,225928  ,467.8,467.1,467.1
XS GIS Cut Line= 4
2306408.03160126626966.4290046142306702.58970084627185.357321875
2307132.48530565627288.8507082162307462.86803897627471.954391743
#Sta/Elev= 30
       0 3464.64    10.6 3455.99      50 3431.37    99.9 3405.71   119.8 3397.26
   134.7 3385.86   170.7 3363.24   272.8 3305.32   299.2 3290.86   324.1 3281.36
   359.4 3264.65   413.9 3248.28   492.1 3238.57   533.2 3237.34     562 3224.95
     587 3222.31   590.3 3222.02   683.2 3222.52     706 3227.29   738.9 3242.49
     776 3246.08   784.2 3251.39   800.6 3257.11   900.4 3283.26  1037.5 3352.24
  1106.9 3379.09  1124.4 3383.76  1156.4 3395.78  1174.1 3403.78  1186.9 3412.48
#Mann= 3 ,-1,0
       0      .1       0     587    .045       0   683.2      .1       0
Bank Sta=587,683.2
XS Rating Curve= 0 ,0
Exp/Cntr(USF)=0,0
Exp/Cntr=0.3,0.1

Type RM Length L Ch R = 1 ,225461  ,558,546.8,543.9
XS GIS Cut Line= 2
2306230.98144007627551.9792904232307247.75473648627796.698204226
#Sta/Elev= 30
       0 3376.19    45.1 3364.25   104.1 3343.53   147.9 3319.89   198.7 3301.26
   235.7 3280.54   256.3 3271.93   272.8 3262.42   285.1 3258.11   309.8 3244.82
   330.4  3238.4   355.1 3234.06   523.7  3233.2   548.4 3227.07   564.9 3219.39
   572.4 3219.18   677.3 3219.32   692.4  3223.6     713 3237.16   729.4 3240.53
   745.9 3239.46     750 3241.21   766.5 3254.13   778.8 3266.94   799.4 3280.02
   906.4 3331.67     957 3351.21   972.2 3358.76  1005.1 3379.17  1045.8 3397.98
#Mann= 5 ,-1,0
       0      .1       0     430     .12       0     530      .1       0
   564.9    .045       0   677.3      .1       0
Bank Sta=564.9,677.3
XS Rating Curve= 0 ,0
Exp/Cntr(USF)=0,0
Exp/Cntr=0.3,0.1

Type RM Length L Ch R = 1 ,224914  ,457.1,441.2,433.2
XS GIS Cut Line= 3
 2306041.8242342628152.6224326812306825.98566148628236.213244726
2307184.31560014628131.226952492
#Sta/Elev= 30
       0 3378.42    30.5 3366.42   139.1 3340.14   247.7 3305.22   315.3 3286.78
   380.5  3265.1   404.6 3254.07     473 3236.12   541.4 3225.88   551.6 3221.56
   561.5 3214.71   569.4 3214.56   672.9 3214.72   718.4 3221.58   738.5 3235.28
   770.7 3238.11   799.1 3264.44   831.5 3282.92   844.4 3297.41   870.5 3310.85
   953.4 3346.16   965.9  3356.2   976.6 3359.92   978.5 3361.62   986.8 3376.41
   999.3 3384.67  1007.6 3387.28    1066 3394.39  1141.1 3406.49    1162 3411.41
#Mann= 3 ,-1,0
       0      .1       0   561.5    .045       0   672.9      .1       0
Bank Sta=561.5,672.9
XS Rating Curve= 0 ,0
Exp/Cntr(USF)=0,0
Exp/Cntr=0.3,0.1

Type RM Length L Ch R = 1 ,224473  ,498.9,490.4,485.3
XS GIS Cut Line= 3
2306101.53195709628741.7386318552306849.86875064628630.284215795
2307243.93972171628351.648175645
#Sta/Elev= 30
       0 3422.46    22.9 3413.46    55.2 3395.53      88 3374.92   111.9 3364.67
     120 3359.51   242.2 3320.58   386.5 3260.17   419.2 3252.42   451.6 3239.19
   479.9 3232.64     488 3229.22   504.1 3228.57   528.4 3214.58   540.5 3210.12
   611.8 3210.07   613.3 3210.08   641.6 3216.58     661 3225.64   694.2 3227.93
   713.8 3233.96   742.7  3235.3   746.8  3236.8   759.4 3249.11   813.9 3272.74
     877 3290.86   960.3 3309.38  1063.1 3336.62  1137.8  3362.1  1239.2 3391.31
#Mann= 6 ,-1,0
       0      .1       0   540.5    .045       0   613.3      .1       0
  886.59     .12       0 1056.59      .1       0 1106.59     .12       0
Bank Sta=540.5,613.3
XS Rating Curve= 0 ,0
Exp/Cntr(USF)=0,0
Exp/Cntr=0.3,0.1

Type RM Length L Ch R = 1 ,223983  ,409.5,403.4,408.7
XS GIS Cut Line= 3
2306435.89520527629259.2055635612307100.64118677629024.355186864
2307554.41988073629060.179820597
#Sta/Elev= 30
       0  3429.7    33.2 3405.26    67.6 3371.03    80.9 3364.63   131.8 3331.66
   161.7 3319.43   240.1 3276.95     276  3253.9   340.4 3224.01   356.6 3219.39
   382.1 3206.54   386.3 3206.27     450  3206.4   462.7 3209.82   496.6  3211.7
   558.4 3227.29   585.7 3228.22   594.3 3230.25   611.2 3229.24   619.7 3231.46
   640.9 3231.45   674.8  3235.5   708.6 3243.15   720.6 3248.76   728.6 3249.43
   784.8 3264.32   804.9 3273.22   828.9 3280.55  1061.7 3328.79  1160.2 3366.95
#Mann= 5 ,-1,0
       0      .1       0     330    .025       0   382.1    .045       0
     450      .1       0 1015.01     .12       0
Bank Sta=382.1,450
XS Rating Curve= 0 ,0
Exp/Cntr(USF)=0,0
Exp/Cntr=0.3,0.1

Type RM Length L Ch R = 1 ,223579  ,676.4,744,830
XS GIS Cut Line= 4
2306495.60292816629394.5430687772306798.12205747629565.705207726
 2307196.1735434629402.504098496 2307626.0691482629402.504098496
#Sta/Elev= 30
       0 3406.17      20 3402.26    40.5 3393.52     108 3357.19   179.9 3331.68
   254.8 3312.75   340.8 3281.35   367.1 3275.27   395.6 3264.56   436.3 3245.65
   457.9 3232.62   483.8 3223.45   518.4 3217.51   548.9 3207.11   585.6 3205.23
   656.2 3204.57   665.4 3205.34   665.4 3205.35   678.4 3212.28   691.3  3222.2
   725.9 3226.52   743.2  3226.3   760.4 3236.87   829.8 3256.11   860.5 3267.19
   925.8 3294.91  1048.5 3331.15  1124.5 3356.19  1149.8 3362.25  1207.7 3382.32
#Mann= 7 ,-1,0
       0      .1       0     300     .12       0  397.58      .1       0
   585.6    .045       0   665.4      .1       0  917.79     .12       0
 1117.79      .1       0
Bank Sta=585.6,665.4
XS Rating Curve= 0 ,0
Exp/Cntr(USF)=0,0
Exp/Cntr=0.3,0.1

Type RM Length L Ch R = 1 ,222835  ,471.9,481.9,488.4
XS GIS Cut Line= 4
2306447.83674985  629490.07542542306849.86875064629848.321762735
 2306941.4205924630198.6070703522307032.97243416630329.964060709
#Sta/Elev= 30
       0  3391.6    19.4 3382.88    34.7 3373.05    76.1 3352.01   112.9 3337.44
   172.4 3317.97   220.6 3306.65   245.2 3294.09   287.3 3278.34   365.4 3263.97
   407.6 3259.71   504.1 3246.17   551.8 3236.13   622.1 3214.53   667.5 3209.13
   688.2 3208.34   718.1  3199.3   816.4 3199.12   832.9 3203.04   857.7 3219.03
   870.1  3220.6   878.4 3228.73   908.6 3250.16   947.3 3285.41   961.8  3296.2
   971.9 3302.19   981.7 3305.62   993.4 3313.94  1042.3 3339.07  1060.7 3350.88
#Mann= 5 ,-1,0
       0      .1       0     380     .12       0  628.49    .025       0
   718.1    .045       0   816.4      .1       0
Bank Sta=718.1,816.4
XS Rating Curve= 0 ,0
Exp/Cntr(USF)=0,0
Exp/Cntr=0.3,0.1

Type RM Length L Ch R = 1 ,222353  ,536.4,540,541.6
XS GIS Cut Line= 4
  2306189.103284629609.4908711782306412.01211612629927.932059921
2306455.79777957630325.9835458492306571.23271049630497.145684798
#Sta/Elev= 30
       0 3392.42    63.1 3360.06     107  3332.8   116.9 3330.11   165.6 3309.42
   180.1 3307.56   292.6 3258.96   340.9 3246.87   368.1 3242.73   414.1 3231.76
   462.4 3227.21   491.5 3222.08     503 3217.14   522.8 3204.13     559 3198.06
   687.3 3198.03   695.8 3200.27     709 3210.37   719.9 3216.16   744.1 3214.79
   760.2 3220.21     797 3242.25     835 3270.75   847.1 3287.73   855.7 3296.89
   897.1  3315.6   928.1 3322.46   961.9 3340.42   981.2  3355.2   995.6 3361.76
#Mann= 6 ,-1,0
       0      .1       0     160     .12       0     280      .1       0
  498.71     .05       0     559    .045       0   687.3      .1       0
Bank Sta=559,687.3
XS Rating Curve= 0 ,0
Exp/Cntr(USF)=0,0
Exp/Cntr=0.3,0.1

Type RM Length L Ch R = 1 ,221813  ,691.9,653.9,605.6
XS GIS Cut Line= 4
2305723.38304546629740.8478615352305886.58415469630003.561842247
2305914.44775871630401.6133281762306161.23967998630616.561130577
#Sta/Elev= 30
       0    3414    66.3  3372.7    79.2 3367.52    89.9 3361.04   107.6 3344.96
   127.5  3332.6     282 3253.76   312.3 3241.67     359 3228.95   399.9 3220.11
   415.2 3212.82   427.2 3209.75   435.2 3204.01   443.2 3194.54   446.6 3194.02
   447.2 3193.94   583.6 3193.94   603.6 3200.18   619.7  3208.2   659.8  3210.8
   671.8 3213.21   683.8 3211.82   687.8 3213.33   699.8 3226.03     732  3241.3
   829.4 3275.95   933.4 3302.81    1000 3329.59  1012.9 3336.17  1035.6 3342.36
#Mann= 4 ,-1,0
       0      .1       0  439.28    .025       0   446.6    .045       0
   583.6      .1       0
Bank Sta=446.6,583.6
XS Rating Curve= 0 ,0
Exp/Cntr(USF)=0,0
Exp/Cntr=0.3,0.1

Type RM Length L Ch R = 1 ,221159  ,492.2,477.9,458.8
XS GIS Cut Line= 2
2304935.24110332630138.899347463 2305846.7790061630863.353051852
#Sta/Elev= 30
       0 3419.81    67.8 3402.41   118.7 3377.49   138.9 3364.63   190.2 3347.75
   241.5 3323.54   357.3 3255.87   372.4 3242.88   386.6 3225.95   403.7 3208.51
   435.5 3186.25   440.6 3185.97   522.4 3186.14   548.9 3192.75   563.2 3199.05
   597.3 3200.09   624.5 3198.13     677 3200.85   696.9 3197.92   716.5 3198.05
     743 3205.69   765.2  3208.2   779.5 3206.43   820.1    3214   913.3 3243.44
   982.2 3259.44  1043.5 3277.29  1084.4 3289.78  1129.6 3307.26  1164.4  3317.3
#Mann= 3 ,-1,0
       0      .1       0   435.5    .045       0   522.4      .1       0
#XS Ineff= 2 , 0
                          591.77         3227.07
Permanent Ineff=
       F       F
Bank Sta=435.5,522.4
XS Rating Curve= 0 ,0
Exp/Cntr(USF)=0,0
Exp/Cntr=0.3,0.1

Type RM Length L Ch R = 1 ,220682  ,436,429,422.6
XS GIS Cut Line= 3
2304678.58064495630717.3178065432305420.61481475630957.061502412
2305752.49045396631110.144973128
#Sta/Elev= 30
       0 3442.98    73.1 3407.89   115.2 3395.25   136.2 3385.36     153 3359.18
   156.8 3355.27   169.8 3346.82   182.4 3343.67   203.4  3327.8   216.1 3322.27
   253.9 3291.03   304.3 3253.35   329.6 3223.83   350.8 3203.28   384.2 3183.85
   480.9 3183.56   485.1 3183.64   515.8 3197.68   601.6 3197.28   615.4 3194.55
   640.6 3194.55   652.5 3196.58     670 3203.84   695.3 3202.12   754.1  3210.5
   832.2  3241.4   955.5 3270.78  1064.8 3309.95  1100.9 3319.08  1145.3 3325.58
#Mann= 3 ,-1,0
       0      .1       0   384.2    .045       0   485.1      .1       0
#XS Ineff= 2 , 0
                          537.18         3223.45
Permanent Ineff=
       F       F
Bank Sta=384.2,485.1
XS Rating Curve= 0 ,0
Exp/Cntr(USF)=0,0
Exp/Cntr=0.3,0.1

Type RM Length L Ch R = 1 ,220252  ,500.4,504.7,509
XS GIS Cut Line= 4
 2304497.3844688631110.1449731282304851.65029128631245.482478344
2305233.77971777631305.1902012332305568.14296595631484.313369901
#Sta/Elev= 30
       0 3411.54    41.7 3394.45    80.1 3369.11   131.5 3341.36   165.4 3323.78
   181.1 3318.77     199 3308.19   212.1 3304.15   242.8 3285.48   255.1 3281.64
   324.1 3245.48     337 3241.08     396 3212.34   440.5 3201.11   477.5 3183.13
   545.8 3181.52   553.9 3183.03   590.3 3185.06   618.6 3191.07   642.9  3192.3
     663 3197.73     736 3199.89   752.2 3212.65   764.4  3214.7   836.8 3237.58
     864 3250.99     893 3261.32     951  3278.6  1018.3 3305.11  1145.3 3345.43
#Mann= 3 ,-1,0
       0      .1       0   477.5    .045       0   553.9      .1       0
#XS Ineff= 2 , 0
                          610.83         3213.62
Permanent Ineff=
       F       F
Bank Sta=477.5,553.9
XS Rating Curve= 0 ,0
Exp/Cntr(USF)=0,0
Exp/Cntr=0.3,0.1

Type RM Length L Ch R = 1 ,219748  ,465.9,465.2,465
XS GIS Cut Line= 2
 2304370.0079933 631655.475508852305404.94185672631858.481766673
#Sta/Elev= 30
       0 3360.91    18.5  3354.7    59.3 3333.26   108.2  3313.2   201.9 3279.22
   226.4  3267.1   250.9 3259.51   323.6 3231.32   352.8 3223.77     365 3218.83
   450.6 3201.86   462.8  3195.8   487.3 3194.41   528.1 3179.81   646.3 3179.67
   650.3  3179.7   678.9  3186.4   691.1 3192.78   711.5 3194.96   715.6 3196.79
   731.9 3214.31   752.2 3225.24   817.8 3248.39     846  3265.5   894.9 3289.76
   939.7 3316.65     952 3319.01   972.4 3328.16  1001.8 3338.13  1054.7 3365.12
#Mann= 6 ,-1,0
       0      .1       0     110     .12       0     270      .1       0
   528.1    .045       0   650.3    .025       0     720      .1       0
Bank Sta=528.1,650.3
XS Rating Curve= 0 ,0
Exp/Cntr(USF)=0,0
Exp/Cntr=0.3,0.1

Type RM Length L Ch R = 1 ,219283  ,556.1,548.4,539.9
XS GIS Cut Line= 2
2304234.67048809632121.195747386 2305269.6043515632288.377371476
#Sta/Elev= 30
       0 3412.67    25.8 3400.77    58.2 3378.87    71.1 3375.35   110.9 3346.56
   143.3 3333.01   167.6 3318.96   175.8 3317.62   190.3 3309.59   268.9 3276.29
   289.2 3270.54   345.9 3247.21   443.2  3203.3   459.4 3196.71   516.1 3186.18
   540.4 3179.01   572.8 3175.42   657.9  3175.4     685 3180.96   698.4  3188.8
   714.7 3191.75   730.9  3190.5   759.2 3212.49   811.9 3237.14   866.9 3267.65
   895.8 3290.07   925.3 3308.71   949.7 3320.72   986.1 3342.93  1048.3 3371.26
#Mann= 5 ,-1,0
       0      .1       0   572.8    .045       0   657.9      .1       0
     850     .12       0     950      .1       0
Bank Sta=572.8,657.9
XS Rating Curve= 0 ,0
Exp/Cntr(USF)=0,0
Exp/Cntr=0.3,0.1

Type RM Length L Ch R = 1 ,218734  ,638.6,599.1,560.9
XS GIS Cut Line= 4
2304167.00173548632495.3641441582304441.65726077632758.078124871
2304983.00728163 632762.058639732305305.42898524632578.954956203
#Sta/Elev= 30
       0 3363.22    40.4 3350.93    81.3 3331.64   152.1 3305.34     211 3285.94
     223 3278.08   245.7 3270.66     263 3261.46   274.6 3258.06   330.3 3228.88
   355.8 3218.88   380.1 3204.91   422.6 3206.82   458.6 3204.99   516.7 3196.22
   542.6  3185.1   630.6 3183.36   662.6 3173.05   782.6 3173.03   830.6 3184.93
   858.6 3187.72   874.6 3185.85   906.6 3194.44     932 3204.78  1019.8 3244.42
  1056.2  3265.2    1069 3270.49  1152.8 3320.39  1204.6 3343.64  1292.2 3386.96
#Mann= 3 ,-1,0
       0      .1       0   662.6    .045       0   782.6      .1       0
Bank Sta=662.6,782.6
XS Rating Curve= 0 ,0
Exp/Cntr(USF)=0,0
Exp/Cntr=0.3,0.1

Type RM Length L Ch R = 1 ,218135  ,624.3,584.2,549.3
XS GIS Cut Line= 3
2304465.54034993633661.6549979282305201.93559889 633152.14909594
2305464.64957961 632821.76636262
#Sta/Elev= 30
       0 3396.54    32.4 3374.46    42.5 3371.88    61.6 3359.39   134.4 3321.19
   197.7 3292.18   225.8 3281.39   312.7 3239.71   407.6 3205.65   471.9 3189.86
     514 3182.71   539.9 3169.11   674.4 3168.99     675    3169   679.3 3169.16
   686.5  3175.4   693.9 3176.78     767 3176.15     790 3173.81   841.7 3184.88
     859 3184.63     869 3190.85   896.3 3201.56     935 3213.92  1078.1 3248.17
  1149.7 3274.21    1218 3305.85  1233.3 3315.09    1257  3323.3  1317.6 3352.88
#Mann= 3 ,-1,0
       0      .1       0   539.9    .045       0     675      .1       0
Bank Sta=539.9,675
XS Rating Curve= 0 ,0
Exp/Cntr(USF)=0,0
Exp/Cntr=0.3,0.1

Type RM Length L Ch R = 1 ,217551  ,641.1,626,609
XS GIS Cut Line= 3
2305253.68229206634127.3752364642305544.25987679633327.291749749
2305715.42201574632893.415630087
#Sta/Elev= 30
       0 3379.92     101 3342.02     147 3329.35   240.7 3283.38   283.2 3258.08
   308.7 3238.83   321.5 3232.73   365.8 3201.62     397 3188.55   410.9 3186.05
   419.4 3181.14   436.4 3178.32   457.7 3167.14   470.5  3163.7   565.6 3163.56
   571.8 3163.63   606.6 3168.76   657.7  3180.7   722.1 3183.86   734.3 3187.51
   948.1 3210.68   969.6 3215.87   999.7 3224.48  1072.8 3253.33  1141.6 3289.05
  1184.6 3316.16  1223.3 3334.43  1240.5 3339.88  1296.4  3369.1  1317.6  3376.3
#Mann= 6 ,-1,0
       0      .1       0     170     .12       0     280      .1       0
     380    .025       0   470.5    .045       0   571.8      .1       0
Bank Sta=470.5,571.8
XS Rating Curve= 0 ,0
Exp/Cntr(USF)=0,0
Exp/Cntr=0.3,0.1

Type RM Length L Ch R = 1 ,216925  ,864.4,860.8,864.1
XS GIS Cut Line= 3
2306065.70732336634147.2778107612306013.96063019633295.447630874
2306085.60989765632869.532540931
#Sta/Elev= 30
       0 3366.92    50.2 3358.07    62.2 3352.95    82.3 3335.88   203.7 3294.07
   266.6 3268.22   294.6  3245.4   318.7 3200.52   338.7 3173.76   355.1 3162.59
   370.8 3158.07   434.9 3158.06     499 3166.74   575.2 3168.04   611.2 3165.51
   631.3 3174.85   675.9 3178.73   694.8 3176.93   747.7 3187.22   823.6 3195.71
   888.2 3209.12   924.7 3222.63   989.6 3254.15  1054.5 3294.64  1066.6 3298.97
  1103.1 3320.76  1123.4 3328.53  1187.1 3362.45  1224.8 3376.92  1285.3 3418.15
#Mann= 4 ,-1,0
       0      .1       0     280    .025       0   370.8    .045       0
   434.9      .1       0
Bank Sta=370.8,434.9
XS Rating Curve= 0 ,0
Exp/Cntr(USF)=0,0
Exp/Cntr=0.3,0.1

Type RM Length L Ch R = 1 ,216064  ,813.9,813.1,815.4
XS GIS Cut Line= 2
2306794.14154261634031.8428798422306893.65441409632969.045412413
#Sta/Elev= 30
       0 3297.14    95.1  3255.6   199.5 3218.89   239.7 3206.04   283.9 3194.55
   323.9 3180.36   356.2 3173.02   428.5 3163.92   480.8 3153.39   522.3 3152.83
     537 3150.34   581.2 3150.31   585.2 3150.81   597.3 3157.43   617.4 3170.89
   641.5 3173.14   653.5 3179.88   697.7 3192.58   721.8 3202.14   818.2 3247.46
   830.3 3255.71   842.3 3261.22   934.7 3285.12   950.8 3294.07   962.9 3297.94
     987 3313.65    1003 3320.02  1027.1 3336.74  1043.2 3343.14  1067.4 3357.17
#Mann= 5 ,-1,0
       0      .1       0     460    .025       0     490      .1       0
     537    .045       0   581.2      .1       0
Bank Sta=537,581.2
XS Rating Curve= 0 ,0
Exp/Cntr(USF)=0,0
Exp/Cntr=0.3,0.1

Type RM Length L Ch R = 1 ,215251  ,680.5,667.6,651.6
XS GIS Cut Line= 2
2307450.92649439634278.6348011172307769.36768313633195.934759392
#Sta/Elev= 30
       0 3315.65    59.9 3293.42   130.8 3258.76   189.1 3240.23   259.9  3210.8
   287.9 3202.76   347.6 3191.11   376.8 3188.93   422.6 3171.22   456.5 3163.32
   501.6 3145.95   501.8 3145.93   651.9 3146.01   656.1 3147.37   664.5 3157.67
   685.2 3167.25     727 3169.96   756.1 3189.68   793.7 3209.95   864.6  3243.9
   872.9 3245.39     923 3267.57     948 3283.47   968.7 3286.59     998 3298.14
  1010.6 3304.34  1035.5 3322.65  1043.9 3325.09  1077.2 3345.27  1128.6 3369.24
#Mann= 4 ,-1,0
       0      .1       0   501.6    .045       0   651.9    .025       0
     740      .1       0
Bank Sta=501.6,651.9
XS Rating Curve= 0 ,0
Exp/Cntr(USF)=0,0
Exp/Cntr=0.3,0.1

Type RM Length L Ch R = 1 ,214584  ,546.9,534.2,517.9
XS GIS Cut Line= 2
2308239.06843653634286.5958308362308266.93204054633219.817848548
#Sta/Elev= 30
       0 3327.87    37.6 3303.91    73.4 3285.58   133.5 3240.45   185.7 3205.87
   249.5  3173.3   277.5 3156.88   289.5 3154.82   312.6 3143.16   321.5 3139.66
   409.6 3139.84   425.6 3143.31   433.6 3144.66   469.6 3159.93   489.6 3164.92
   505.6 3174.09   513.3 3173.53   528.9 3166.59   552.3 3166.04   569.6  3178.4
   614.7 3187.97   793.7 3238.57   897.7  3261.7   917.7 3269.25   937.7 3282.23
   961.7 3290.91   989.8 3298.09  1025.8  3310.9  1033.8 3311.13  1067.1 3319.47
#Mann= 3 ,-1,0
       0      .1       0   312.6    .045       0   425.6      .1       0
Bank Sta=312.6,425.6
XS Rating Curve= 0 ,0
Exp/Cntr(USF)=0,0
Exp/Cntr=0.3,0.1

Type RM Length L Ch R = 1 ,214049  ,605.2,640.2,666.2
XS GIS Cut Line= 3
2308852.06772486634147.277810761 2308700.8081602633578.064185883
2308661.00301161633136.227036503
#Sta/Elev= 30
       0 3339.26     6.3 3338.45    10.4 3335.16    31.1 3313.25    89.1 3276.66
   113.9 3249.58   142.2 3224.34   155.3 3213.03   184.3 3194.28   233.9 3151.21
   246.4 3147.27   258.8 3137.13   262.9    3136   349.8    3136   387.5 3149.14
   411.9 3152.51   432.6 3158.24   462.7 3161.84   478.1 3160.69   494.7 3166.72
   515.4  3167.4   560.3 3174.12     614 3187.53   664.3 3202.48   774.6 3244.41
   826.8 3261.37     879 3282.56   951.4 3315.73  1003.5 3332.78  1032.6 3347.05
#Mann= 4 ,-1,0
       0      .1       0     190    .025       0   262.9    .045       0
   349.8      .1       0
Bank Sta=262.9,349.8
XS Rating Curve= 0 ,0
Exp/Cntr(USF)=0,0
Exp/Cntr=0.3,0.1

Type RM Length L Ch R = 1 ,213409  ,458.1,483,512.6
XS GIS Cut Line= 3
2308887.89235859634139.3167810422309182.45045818633912.427434063
2309652.15121157633402.921532075
#Sta/Elev= 30
       0 3314.62    10.5 3307.47    55.9  3290.9   121.5 3277.88   146.8 3263.63
   164.3 3250.72   219.8  3231.7   252.7 3225.75   338.6 3221.58     344  3218.4
   353.8 3205.62   392.6 3192.43   417.8 3174.72   480.6 3149.15   566.6 3145.49
   579.1 3142.01   590.5 3135.54   607.5 3132.51   615.6 3130.25   669.7    3132
   687.1 3133.84   702.7 3142.28     719  3155.3   754.7 3159.01     783 3182.65
   822.9 3207.12   838.7 3219.98  1007.3 3299.26  1026.4 3311.02  1064.8 3328.51
#Mann= 7 ,-1,0
       0      .1       0      30     .12       0     120      .1       0
  571.81    .025       0   607.5    .045       0   669.7    .025       0
  691.81      .1       0
Bank Sta=607.5,669.7
XS Rating Curve= 0 ,0
Exp/Cntr(USF)=0,0
Exp/Cntr=0.3,0.1

Type RM Length L Ch R = 1 ,212926  ,527.4,526.1,530.3
XS GIS Cut Line= 3
2308867.98978429634191.0634742132309309.11798289634107.075464252
2309971.58710339634179.538233691
#Sta/Elev= 30
       0 3337.83    28.7 3322.15    40.9  3312.9    77.6 3296.93   155.7 3276.74
   191.6 3256.51     216 3249.66   277.1 3226.56   309.7 3217.29   346.3 3195.23
   358.5 3190.73   370.7 3182.85   403.3 3170.92   464.6 3155.58   548.7  3149.4
   568.8 3140.37   580.7 3137.91   660.5 3129.55     704 3129.42   716.7 3129.46
   733.8 3136.81   753.9 3150.55     770 3152.22   810.3 3184.67   890.7  3233.1
   936.1 3257.39   967.2  3270.9  1055.5 3321.88    1100 3343.61  1115.5 3353.13
#Mann= 4 ,-1,0
       0     .12       0      40      .1       0   660.5    .045       0
   716.7      .1       0
Bank Sta=660.5,716.7
XS Rating Curve= 0 ,0
Exp/Cntr(USF)=0,0
Exp/Cntr=0.3,0.1

Type RM Length L Ch R = 1 ,212400  ,440.9,438.4,439.8
XS GIS Cut Line= 3
2308800.32103169634509.5046629552309572.54091439634676.686287045
2309863.11849911634684.647316764
#Sta/Elev= 30
       0 3365.32    70.3 3332.59    89.9 3317.88   102.2 3312.06   114.4 3300.42
   179.9 3264.62   216.8 3238.97   249.5 3227.96   306.8 3200.08   335.4 3182.46
   347.7 3178.62   388.7  3152.4   433.7 3136.12   544.2 3139.71   556.5 3131.63
   568.7 3127.49   697.9 3127.55   716.1 3131.35   736.5 3143.81   765.2 3146.57
   769.3 3148.47   785.6 3166.06   809.8 3174.92   837.8 3179.59   869.8    3202
   945.8 3226.06   969.8 3228.07   993.8 3239.89  1045.8 3255.99  1080.8 3280.85
#Mann= 6 ,-1,0
       0      .1       0   568.7    .045       0   697.9      .1       0
     710    .025       0     720      .1       0  920.11     .12       0
Bank Sta=568.7,697.9
XS Rating Curve= 0 ,0
Exp/Cntr(USF)=0,0
Exp/Cntr=0.3,0.1

Type RM Length L Ch R = 1 ,211962  ,376.1,374,371.8
XS GIS Cut Line= 2
2308840.12618028635026.971594662 2309707.8784196635082.698802692
#Sta/Elev= 30
       0 3317.46     8.1  3310.3    52.2 3279.88    80.2  3265.6   132.3 3231.41
   180.4 3204.27   268.6 3168.18   295.9 3154.21   340.7 3134.56   364.8 3133.17
   380.8 3127.64   396.9 3124.88   420.9 3124.87   464.6 3124.91     477 3126.72
   545.2 3126.88   561.2  3133.1   577.2 3136.92   589.7  3143.6   613.3 3143.59
   661.4 3174.77   665.4 3178.86   673.4 3192.25   677.4  3196.1   683.8 3198.34
   709.5 3201.84   725.5 3212.59   809.7 3242.77   829.8 3253.97   869.5 3271.65
#Mann= 3 ,-1,0
       0      .1       0   396.9    .045       0   464.6      .1       0
Bank Sta=396.9,464.6
XS Rating Curve= 0 ,0
Exp/Cntr(USF)=0,0
Exp/Cntr=0.3,0.1

Type RM Length L Ch R = 1 ,211588  ,457.2,451.7,449.1
XS GIS Cut Line= 2
2308796.34051683635417.0620508722309731.76150876635436.964625168
#Sta/Elev= 30
       0 3317.98    51.8 3277.66   135.9 3230.91   163.9 3211.26   187.9 3198.08
   295.9 3152.78   315.9 3142.06     339    3135   355.9 3132.53   371.9  3124.1
   391.9 3121.75   475.9 3121.84   539.3 3129.24   552.3 3132.78     568 3140.44
     588 3139.76     600 3142.33     640 3158.95     652 3161.44     668 3169.79
     708 3181.05     728 3190.99     752 3193.19     768  3201.8   825.5 3220.42
     840 3228.63   862.3 3233.81     888 3243.51     912  3255.3   935.6 3271.43
#Mann= 7 ,-1,0
       0      .1       0   391.9    .045       0   475.9      .1       0
     510     .12       0     610      .1       0     710     .12       0
     800      .1       0
Bank Sta=391.9,475.9
XS Rating Curve= 0 ,0
Exp/Cntr(USF)=0,0
Exp/Cntr=0.3,0.1

Type RM Length L Ch R = 1 ,211136  ,903.3,921.3,946.2
XS GIS Cut Line= 3
2308887.89235859635894.7238339862309457.10598347635866.860229971
 2309835.2548951635711.620150459
#Sta/Elev= 30
       0 3265.15    24.3 3261.66    32.3 3250.31    36.3 3246.91    68.4 3230.28
    76.4 3224.88    88.4 3213.35   112.4  3197.3   164.5  3175.6   188.2 3163.27
   220.5 3142.87   240.6 3132.79   256.6 3128.54   272.6 3118.91   414.1 3118.76
   416.8 3118.83   436.8 3125.52   472.8 3126.26   504.9 3140.66   520.9 3137.06
   548.9 3137.53   573.2 3151.77   586.2 3165.49   603.5 3167.86   628.7 3175.16
   733.2 3198.22     824 3225.15   880.2 3253.29   932.1 3269.39   978.7 3287.26
#Mann= 8 ,-1,0
       0      .1       0     120     .12       0     220      .1       0
   272.6    .045       0   416.8      .1       0     420    .025       0
     520      .1       0   939.9     .12       0
Bank Sta=272.6,416.8
XS Rating Curve= 0 ,0
Exp/Cntr(USF)=0,0
Exp/Cntr=0.3,0.1

Type RM Length L Ch R = 1 ,210215  ,819.3,853,889.3
XS GIS Cut Line= 2
2308692.84713049636145.4962701212309520.79422122636901.794093384
#Sta/Elev= 30
       0 3231.19    20.8 3226.65   112.9 3215.23   188.7 3193.76   253.7 3170.16
   286.2 3161.07     373 3145.25   573.4 3121.09   707.1 3123.62   741.3 3120.75
   770.5 3123.27   782.4 3120.96   794.9  3114.2   812.1 3114.01     828 3110.73
   831.7 3110.72   896.8 3110.76   922.3  3126.1   941.8 3127.87     945 3131.01
   954.4 3146.54   978.1  3204.4   984.6 3216.18  1013.7 3231.18  1035.6 3245.04
  1046.9 3256.13  1061.2 3264.43  1075.2 3277.72  1098.9  3279.2  1121.4 3275.14
#Mann= 3 ,-1,0
       0      .1       0     828    .045       0   896.8      .1       0
#XS Ineff= 2 , 0
          771.99 3134.76
Permanent Ineff=
       F       F
Bank Sta=828,896.8
XS Rating Curve= 0 ,0
Exp/Cntr(USF)=0,0
Exp/Cntr=0.3,0.1

Type RM Length L Ch R = 1 ,209362  ,621.3,607,580.8
XS GIS Cut Line= 3
 2308378.3864566636252.9701713212308529.64602125636563.450330345
 2308505.7629321637176.449618675
#Sta/Elev= 30
       0 3238.87    34.4 3227.93    76.3 3209.91    95.4 3205.03   138.2 3198.62
   147.1 3195.08     175 3189.03   252.8  3157.1   305.5    3148   375.4 3130.95
   447.2 3122.81   483.2 3115.78   495.2  3111.5   511.2 3111.04   519.2 3115.29
   523.2 3115.15   535.2 3111.66   547.2 3111.59   578.9 3104.81   579.3 3104.75
   710.6 3104.89   715.4    3106   735.4 3120.13   751.4 3123.19   767.4 3122.72
   803.1 3154.05   823.5 3167.22   879.5 3213.16   915.5 3230.88   958.8  3248.3
#Mann= 4 ,-1,0
       0      .1       0  515.37    .025       0   578.9    .045       0
   710.6      .1       0
Bank Sta=578.9,710.6
XS Rating Curve= 0 ,0
Exp/Cntr(USF)=0,0
Exp/Cntr=0.3,0.1

Type RM Length L Ch R = 1 ,208755  ,648,623.6,591.3
XS GIS Cut Line= 3
2307681.79635623636599.2749640792308131.59453533637096.839321489
2308374.40594174637196.352192971
#Sta/Elev= 30
       0 3257.29       8  3251.8    21.4 3247.39    51.1 3221.77    67.3 3211.79
      88 3194.36   115.8 3164.27   122.8 3160.14   164.3 3150.27   206.9  3152.4
   249.4 3147.27   255.1 3143.86   272.2 3125.14   301.8 3103.59   309.9 3100.45
     340 3098.59   345.7 3098.55     391 3098.59     442 3107.07   486.7 3106.75
     504 3111.68   617.3  3107.4   640.2 3119.52   660.1 3120.26   683.7 3137.12
   744.4  3174.1   821.7 3197.93   887.5 3228.32   917.8 3238.49   933.1 3239.84
#Mann= 3 ,-1,0
       0      .1       0     340    .045       0     391      .1       0
Bank Sta=340,391
XS Rating Curve= 0 ,0
Exp/Cntr(USF)=0,0
Exp/Cntr=0.3,0.1

Type RM Length L Ch R = 1 ,208131  ,414.3,401.4,389.8
XS GIS Cut Line= 3
2307343.45259319637455.0856588252308016.15960441637355.572787343
2308338.58130801637279.943005016
#Sta/Elev= 30
       0 3326.68    16.9  3312.8    73.5 3275.51    98.3 3261.48   126.1 3239.07
   146.3 3226.62   178.6 3202.66   198.9 3191.57   259.5 3153.49   312.1 3108.43
   328.3 3096.99     341 3092.78   344.4 3092.62   405.1 3092.68   445.5 3095.75
   473.8 3104.74   562.8 3105.28   619.4 3109.94   639.6 3116.54   667.9 3119.47
     680 3118.18   692.4 3126.83   721.1 3133.89   737.6 3140.81   770.4 3150.45
   819.7 3171.09   852.6 3179.74   864.9 3180.89   938.9 3197.97  1011.2 3223.52
#Mann= 3 ,-1,0
       0      .1       0     341    .045       0   405.1      .1       0
Bank Sta=341,405.1
XS Rating Curve= 0 ,0
Exp/Cntr(USF)=0,0
Exp/Cntr=0.3,0.1
