HEC-RAS study SHAVERSFK.prj: SHAVERSFK

--- SHAVERSFK.g01 (geometry) --- (continued)

Type RM Length L Ch R = 1 ,180619  ,305.6,307.1,311.4
XS GIS Cut Line= 2
2318697.04317673648085.6826112642319632.06611717648050.216223868
#Sta/Elev= 30
       0 3101.98    15.1 3093.59    59.2 3060.34    99.2 3002.16   123.2 2961.34
   155.2 2922.05   188.6 2895.19   223.3 2877.17   315.4 2838.13   327.4 2825.43
   339.4 2819.18   427.4  2818.9   447.9  2819.1   483.5 2824.73   499.5 2833.91
   531.1  2835.8   551.9 2842.13   599.6 2868.34   623.6 2888.13     631 2890.95
   651.6 2893.91   663.6 2892.52   678.4 2899.32   695.6  2903.5   751.7 2911.69
   795.7 2922.75   840.4 2927.34   879.8  2928.1   919.8 2938.38   935.7 2945.59
#Mann= 3 ,-1,0
       0      .1       0   339.4    .045       0   447.9      .1       0
Bank Sta=339.4,447.9
XS Rating Curve= 0 ,0
Exp/Cntr(USF)=0,0
Exp/Cntr=0.3,0.1

Type RM Length L Ch R = 1 ,180312  ,324.3,328.6,333.9
XS GIS Cut Line= 2
2318664.98140832648325.9333913812319588.61485816648429.707662477
#Sta/Elev= 30
       0  3041.7    27.4 3035.55    72.5  3011.8    87.7 2994.45     124 2972.54
   144.1 2952.97   156.2  2947.4   188.4 2915.09   226.6  2886.7   255.5 2853.58
   280.8 2833.35   331.5 2818.23   369.5 2818.64   393.7 2822.89426.10532813.079
   482.2 2812.75484.67652812.998   522.5 2817.36   542.6 2834.89   586.9 2859.73
   624.6 2885.96   651.3 2890.26   679.4 2889.76   703.6 2907.53   743.8  2912.5
     768 2921.64   832.4 2958.01   861.5 2981.99   888.8 3000.28   929.4 3031.43
#Mann= 3 ,-1,0
       0      .1       0426.1053    .045       0484.6765      .1       0
Bank Sta=426.1053,484.6765
XS Rating Curve= 0 ,0
Exp/Cntr(USF)=0,0
Exp/Cntr=0.3,0.1

Type RM Length L Ch R = 1 ,179983  ,316.8,317.4,317.5
XS GIS Cut Line= 3
2318593.86823157648578.9878177752319299.97176246648759.543971792
2319441.83731205648811.131444368
#Sta/Elev= 30
       0 3003.91    27.2 2998.55    39.5 2993.53    56.1 2976.88     118 2941.94
   151.7 2919.37   188.2 2889.61   234.9 2862.15   299.6 2817.28   307.9 2815.74
   325.9 2819.13   369.8  2819.7   390.5 2814.59   444.2 2813.41   456.5 2810.26
   466.1 2810.21   530.9 2810.22   551.5 2820.56     568 2836.79   575.8 2841.74
   605.2 2859.14   617.6 2863.56   646.5 2882.61     663 2885.45   691.9 2884.08
   733.3 2900.48   780.2 2927.27   818.4 2961.95   835.4 2974.38   879.8 2985.89
#Mann= 3 ,-1,0
       0      .1       0   456.5    .045       0   530.9      .1       0
Bank Sta=456.5,530.9
XS Rating Curve= 0 ,0
Exp/Cntr(USF)=0,0
Exp/Cntr=0.3,0.1

Type RM Length L Ch R = 1 ,179666  ,407.7,363.7,355.8
XS GIS Cut Line= 2
 2318461.6753331648865.9431339812319277.40224321649081.965675394
#Sta/Elev= 30
       0  2983.6    39.8 2964.72    56.4 2952.78   122.6 2918.32   158.5 2896.19
   168.3 2893.42   197.1 2876.67     284 2843.07   300.5 2824.95   317.1 2810.14
   325.3 2808.28   350.2 2808.19     375  2811.5   424.6 2814.19   461.9 2813.37
   482.3  2809.2   554.3  2809.2   569.5  2815.6     586 2825.63   619.1 2850.97
   652.5 2858.71   677.1 2876.55   688.4 2881.61   697.8  2882.9   718.4 2877.47
   743.3 2882.89     780  2922.9   801.2 2940.24   817.7 2947.29   843.8 2951.85
#Mann= 5 ,-1,0
       0      .1       0     300    .025       0     400      .1       0
   482.3    .045       0   554.3      .1       0
Bank Sta=482.3,554.3
XS Rating Curve= 0 ,0
Exp/Cntr(USF)=0,0
Exp/Cntr=0.3,0.1

Type RM Length L Ch R = 1 ,179302  ,516.1,470.7,438.7
XS GIS Cut Line= 2
 2318310.1371324649243.1765271952319161.33042991649375.369425672
#Sta/Elev= 30
       0 3005.83    46.6 2978.13   107.3 2945.33   147.8 2919.04   155.9  2915.4
   200.4 2887.44   238.3 2868.79   301.4 2831.51   317.8 2823.51   330.7 2820.04
   342.1 2813.73   350.2 2807.02   358.3  2804.6   381.9 2803.65   532.3 2804.94
   560.6 2813.94   609.3 2811.93   625.4 2816.54   641.6  2824.4   657.8 2838.25
   678.1 2853.64   714.5 2879.49   742.8 2882.38     755 2880.91     759 2883.15
   771.2 2892.51   795.5  2918.8   807.6 2929.04     844  2935.7   861.4 2937.05
#Mann= 4 ,-1,0
       0      .1       0     350    .025       0   358.3    .045       0
   532.3      .1       0
Bank Sta=358.3,532.3
XS Rating Curve= 0 ,0
Exp/Cntr(USF)=0,0
Exp/Cntr=0.3,0.1

Type RM Length L Ch R = 1 ,178831  ,503.4,473.8,454.1
XS GIS Cut Line= 2
2318410.08786052650000.8675306592319174.22729806 649465.64750268
#Sta/Elev= 30
       0 3033.88    75.9 2986.17     111 2965.74   139.3 2952.59   215.6 2905.18
   256.9 2876.36   339.5 2812.14   349.3 2806.86   359.1 2804.29   414.8 2799.22
   417.7 2799.09   495.8 2799.09   536.3 2805.13   603.2  2805.2   622.8 2808.82
     636 2808.33   656.9 2804.02   671.6 2805.64   679.1 2810.69   705.8 2834.32
   736.5 2851.11   750.9 2863.23   793.9 2891.49   805.4 2891.99   836.1 2880.09
   857.1 2880.23   896.2 2920.15   901.1 2922.86   919.8 2926.02   932.9 2931.11
#Mann= 3 ,-1,0
       0      .1       0   414.8    .045       0   495.8      .1       0
Bank Sta=414.8,495.8
XS Rating Curve= 0 ,0
Exp/Cntr(USF)=0,0
Exp/Cntr=0.3,0.1

Type RM Length L Ch R = 1 ,178357  ,450.3,433.1,429.9
XS GIS Cut Line= 3
 2319025.9133144650397.4462260892319241.93585581649726.809082598
2319264.50537507649510.786541184
#Sta/Elev= 30
       0 3088.04    29.7 3073.09    42.3  3054.1    59.6 3047.55   109.5 3013.73
   122.2 3007.62   172.6 2972.44   193.6 2951.03   197.8 2941.64   214.6 2896.56
   218.8 2892.07   230.9  2882.8     265 2849.89   307.1 2815.38   333.5 2802.19
   357.5 2795.07   431.1 2795.22   525.6  2802.7   588.6 2801.52   626.4 2795.66
   650.4 2797.04   664.3 2807.01   681.1  2810.7   689.5 2814.67   735.3 2843.83
   770.6  2858.9   794.7 2876.52   838.9 2877.52   867.1 2898.89   921.8 2918.97
#Mann= 3 ,-1,0
       0      .1       0   357.5    .045       0   431.1      .1       0
Bank Sta=357.5,431.1
XS Rating Curve= 0 ,0
Exp/Cntr(USF)=0,0
Exp/Cntr=0.3,0.1

Type RM Length L Ch R = 1 ,177924  ,468.6,501,520.6
XS GIS Cut Line= 2
2319583.70286163650436.1368305222319574.03021052649404.387378996
#Sta/Elev= 30
       0 3103.25      47 3081.58      63 3070.52      87 3047.21     127 3013.07
     147 2986.86     199 2937.91   208.5 2925.01     231 2901.86     263  2873.3
     323 2828.21     355 2800.22     371 2794.84     399 2792.47     411 2786.76
   496.1 2786.56     507 2786.74     531 2790.89     551 2799.74     571 2804.74
     659 2803.96     711 2834.14     775    2854   810.9 2874.76     843 2874.04
     859 2876.57     879    2889     915    2900     959 2911.46  1031.8 2924.52
#Mann= 4 ,-1,0
       0      .1       0     411    .045       0     507    .025       0
     530      .1       0
Bank Sta=411,507
XS Rating Curve= 0 ,0
Exp/Cntr(USF)=0,0
Exp/Cntr=0.3,0.1

Type RM Length L Ch R = 1 ,177423  ,525.1,565.6,593.4
XS GIS Cut Line= 2
2319586.92707867650471.6032179182320425.22350803649678.445827057
#Sta/Elev= 30
       0 3118.23    38.4 3090.04    61.7 3077.54      79 3056.39   194.5 2975.54
   209.2 2963.63   230.5 2938.73     312 2879.27   346.9 2861.13   393.5 2847.54
   429.9  2832.2   492.4 2798.64   574.4 2799.79   585.5 2797.13   601.9 2784.81
   613.8 2780.62     667  2780.5   672.8 2780.67   728.6  2793.5   760.9 2808.57
   789.2 2828.36   833.2 2845.92   857.1 2867.42   888.2 2871.94   917.3 2898.08
   954.4 2909.17   978.8 2910.69  1042.5 2930.25  1075.5 2951.71  1154.1 2962.15
#Mann= 3 ,-1,0
       0      .1       0   613.8    .045       0   672.8      .1       0
Bank Sta=613.8,672.8
XS Rating Curve= 0 ,0
Exp/Cntr(USF)=0,0
Exp/Cntr=0.3,0.1

Type RM Length L Ch R = 1 ,176858  ,410,392.5,382.3
XS GIS Cut Line= 4
2319606.27238088650655.3835889712319996.40264224650523.190690494
2320383.30868656650613.4687675032320573.53749169650552.208643818
#Sta/Elev= 30
       0 3167.51   103.4 3092.78     116 3080.12   128.7 3071.22   149.8 3048.21
   170.9  3034.4     183  3020.6   224.1 2988.48   263.9 2949.45     285 2936.75
   309.2 2917.96   340.8 2888.86     361 2861.67   391.2 2832.31   419.9 2814.73
   440.4 2794.73     460 2780.15   510.3 2772.97   596.7 2773.03   645.8 2784.52
   662.2 2800.51   686.9 2817.98   715.6 2831.48   748.5 2855.48   785.5 2859.56
   801.9 2857.11   826.9 2863.35   852.2 2863.38   924.6 2889.15  1009.1 2913.75
#Mann= 3 ,-1,0
       0      .1       0   510.3    .045       0   596.7      .1       0
Bank Sta=510.3,596.7
XS Rating Curve= 0 ,0
Exp/Cntr(USF)=0,0
Exp/Cntr=0.3,0.1

Type RM Length L Ch R = 1 ,176465  ,480.1,473.4,469.8
XS GIS Cut Line= 3
2319577.25442756650984.2537266452320264.01265623 650922.99360296
2320625.12496427650819.818657808
#Sta/Elev= 30
       0 3187.02      19 3175.31   123.3 3097.14   151.5 3069.53     264 2979.83
   288.1 2965.25   299.7 2954.56   308.1    2945   316.2 2928.33   344.3 2854.06
   376.4  2823.2   432.6 2776.21  437.372769.757   440.7  2767.1   512.9 2767.25
     525 2769.92   593.3 2773.64   613.3 2781.39   625.9 2792.95   689.7 2802.65
   746.1 2821.28   785.3 2847.83   818.6 2850.66   851.9 2869.01   864.4 2869.99
     881 2862.05   901.4 2862.23   918.5 2881.14   922.6  2883.1    1065 2905.41
#Mann= 3 ,-1,0
       0      .1       0  437.37    .045       0     525      .1       0
Bank Sta=437.37,525
XS Rating Curve= 0 ,0
Exp/Cntr(USF)=0,0
Exp/Cntr=0.3,0.1

Type RM Length L Ch R = 1 ,175992  ,389.1,386.8,389.4
XS GIS Cut Line= 3
2319619.16924903651464.662065012 2320028.6448126651432.419894651
2320776.66316496651274.433259886
#Sta/Elev= 30
       0 3101.66    29.1 3085.49    41.1 3063.58    45.1 3059.64    69.2 3045.12
   145.5 2987.39   210.7 2947.72   245.8 2931.21   386.2 2843.54   414.4  2820.2
   438.9  2786.2   455.2 2768.89   463.4 2764.78   483.9 2763.76     492 2762.17
   568.3 2763.91   598.7 2764.85   639.2 2774.75   655.6 2773.39   684.2 2787.63
   741.4 2804.83     815 2812.53   847.7 2834.39   864.1 2839.81   880.4 2837.42
   900.9  2827.9   945.8 2854.29  1007.2    2858  1031.7 2854.14  1175.3 2881.08
#Mann= 3 ,-1,0
       0      .1       0   483.9    .045       0   568.3      .1       0
Bank Sta=483.9,568.3
XS Rating Curve= 0 ,0
Exp/Cntr(USF)=0,0
Exp/Cntr=0.3,0.1

Type RM Length L Ch R = 1 ,175605  ,621,616.6,626.9
XS GIS Cut Line= 2
2319615.94503199651877.3618456222320857.26859086651683.908823461
#Sta/Elev= 30
       0 3075.64   101.4 3011.51   129.8 2982.41   182.4 2943.08   255.3 2910.43
     397 2834.25   433.4 2811.07   473.2 2806.34   546.8    2785     567 2766.33
   583.2 2757.93   627.7 2756.38   631.8 2755.63   690.6  2756.3   704.4  2760.5
   753.2  2786.8   789.6 2796.42   826.1 2818.98   846.3  2819.9   866.6 2827.87
   915.1 2830.46   935.5 2848.08   951.6 2856.86     984 2852.81  1004.2 2860.84
  1064.7 2854.03  1145.9 2854.71  1162.1 2859.38  1202.6 2881.76  1256.3 2899.65
#Mann= 3 ,-1,0
       0      .1       0   627.7    .045       0   690.6      .1       0
Bank Sta=627.7,690.6
XS Rating Curve= 0 ,0
Exp/Cntr(USF)=0,0
Exp/Cntr=0.3,0.1

Type RM Length L Ch R = 1 ,174988  ,480.2,460.7,452.6
XS GIS Cut Line= 3
2319729.32707083 652443.84275115 2320744.4209946652200.081449377
 2320903.2399721652161.241894869
#Sta/Elev= 30
       0 3071.03    54.3 3052.66      77 3051.66   155.1  3015.3   163.4 3002.54
   183.9 2951.81   253.9 2850.74     295 2810.57     332 2756.26   356.7 2747.63
   393.7 2746.17     402 2747.76   488.3 2749.71   505.5  2756.1   570.6 2802.56
   664.7  2815.9   681.7 2824.69   702.3 2819.58   726.9 2826.28   743.4 2817.28
   768.1 2816.67   792.8 2837.24   846.2 2855.68   924.4 2861.45   969.3 2847.95
  1002.6 2863.99  1023.1 2858.16  1084.9 2869.86  1187.8 2931.78  1207.5 2936.18
#Mann= 3 ,-1,0
       0      .1       0   356.7    .045       0     402      .1       0
Bank Sta=356.7,402
XS Rating Curve= 0 ,0
Exp/Cntr(USF)=0,0
Exp/Cntr=0.3,0.1

Type RM Length L Ch R = 1 ,174528  ,618.1,586.4,577.2
XS GIS Cut Line= 3
2320254.34000512653237.9814348222320215.64940069652838.178522355
 2320914.0428661652299.094680858
#Sta/Elev= 30
       0 3126.42    20.9  3113.5      37 3092.88   109.3 3053.59   153.5 3035.42
   173.6 3010.65   221.8  2984.4   245.9 2948.93   303.2 2900.96     350 2845.19
   374.5 2797.09   401.7 2786.35   449.1 2745.58   468.8 2740.24   473.1 2739.86
     564 2740.04   608.1 2750.62   673.7 2750.75   690.8 2757.38   720.7  2777.9
   763.4 2790.62   796.3 2806.16   894.3 2812.56   913.9 2810.03   998.6 2823.07
  1051.4 2821.47  1103.8 2851.66    1143 2846.61  1172.7 2873.48  1283.9 2911.18
#Mann= 4 ,-1,0
       0      .1       0  421.67    .025       0   468.8    .045       0
     564      .1       0
#XS Ineff= 2 , 0
                          621.66         2800.86
Permanent Ineff=
       F       F
Bank Sta=468.8,564
XS Rating Curve= 0 ,0
Exp/Cntr(USF)=0,0
Exp/Cntr=0.3,0.1

Type RM Length L Ch R = 1 ,173941  ,686.3,712,788.6
XS GIS Cut Line= 3
2320657.36713463653366.9501162622321053.94583006652554.447423186
2321057.51174342 652359.71520806
#Sta/Elev= 30
       0 3093.01    46.5 3066.05    66.2 3048.07    77.6 3028.91      91 3022.12
   123.1 2995.69     140 2965.86   180.3 2916.98   202.3 2896.47   218.8 2865.64
   233.4 2850.65   246.8 2829.17   350.4 2746.11   362.4    2741   398.1 2735.84
   411.5  2732.8   487.1 2732.63   504.9 2735.58     545 2764.72   576.2 2779.62
   718.3 2783.23   749.7 2799.13   803.2 2802.26   834.3 2824.98   878.8 2831.39
   909.4 2841.32   941.4 2842.76   957.4 2857.93  1001.8 2887.12  1098.9 2919.06
#Mann= 4 ,-1,0
       0      .1       0   398.1    .045       0   504.9    .025       0
     560      .1       0
Bank Sta=398.1,504.9
XS Rating Curve= 0 ,0
Exp/Cntr(USF)=0,0
Exp/Cntr=0.3,0.1

Type RM Length L Ch R = 1 ,173229  ,347.9,370.3,426.2
BEGIN DESCRIPTION:
Structure XS 4
END DESCRIPTION:
XS GIS Cut Line= 3
2320714.61449471 653480.822801512321105.53330263653512.039882883
2321889.01804239653150.927574849
#Sta/Elev= 30
       0 3041.64    25.6 3021.05    93.9 2977.58   105.9 2961.33   178.1 2918.13
   210.2 2900.78   282.5 2869.85   370.7 2824.36   382.8 2821.26   430.3 2792.64
   456.7 2783.52     541  2779.9   588.9 2771.97   624.1 2749.54   646.1 2727.64
   650.5 2726.74   817.9 2727.81   835.5 2733.96   892.8 2775.78     906 2780.61
     928 2782.19   969.1 2822.79  1002.9 2834.57  1086.6 2844.54  1174.1 2883.54
  1192.3 2897.14  1213.3 2928.05  1218.7 2933.18  1236.3 2947.64  1254.9 2954.42
#Mann= 5 ,-1,0
       0      .1       0  622.16    .025       0   646.1    .045       0
   817.9    .025       0  832.16      .1       0
Bank Sta=646.1,817.9
XS Rating Curve= 0 ,0
Exp/Cntr(USF)=0,0
Exp/Cntr=0.3,0.1

Type RM Length L Ch R = 1 ,172859  ,80.1,83,87.3
BEGIN DESCRIPTION:
Structure XS 3
END DESCRIPTION:
XS GIS Cut Line= 6
2320673.23411583653694.646214873 2321182.9145115653711.941339116
2321563.37212175653757.0803776212321660.09863283653802.219416125
2321698.78923726653840.9100205572321840.65478684653786.098330945
#Sta/Elev= 30
       0 2978.77      31 2960.46      71 2929.06      83  2924.5     111 2900.24
     133 2887.38     171 2871.45   251.1 2849.22     307 2847.44   348.4 2828.43
   395.2 2801.91   435.2  2792.9   481.4 2788.45   535.4 2767.85   587.8 2760.98
     613  2747.5   684.4 2746.88   720.2 2723.11     765 2720.55   820.8 2723.14
   837.5 2734.09   873.8 2765.97   938.1 2770.35   964.6 2789.55   986.7 2798.68
  1050.1 2805.78  1067.8 2814.27  1142.6 2818.77  1185.3  2831.7  1206.6 2832.82
#Mann= 4 ,-1,0
       0      .1       0   720.2    .045       0   820.8    .025       0
  839.97      .1       0
Bank Sta=720.2,820.8
XS Rating Curve= 0 ,0
Exp/Cntr(USF)=0,0
Exp/Cntr=0.3,0.1

Type RM Length L Ch R = 1 ,172776  ,307.5,305.8,314.1
BEGIN DESCRIPTION:
Structure XS 2
END DESCRIPTION:
XS GIS Cut Line= 6
 2320619.4475152653797.6284137742320834.14997798653812.312718243
2321289.31367369653798.9951990892321515.00886621653837.685803521
2321663.32284986653950.5333997822321898.69069349653850.582671665
#Sta/Elev= 30
       0 2980.28    24.8 2965.23    60.9 2933.79     121 2891.87   169.3 2881.66
   217.2 2859.11   325.3 2839.46   377.3  2835.1   389.3 2830.05   413.3  2810.4
   441.3 2792.59   453.2  2791.5   521.4 2769.68   681.9 2764.18   705.9 2757.08
   744.2  2724.7   774.9 2721.04     783 2719.59   837.9 2720.97   858.5 2731.41
     901 2766.08   942.8  2767.9   976.4  2790.7  1006.6 2801.99  1085.9 2796.26
  1112.9 2776.93  1136.4 2773.28  1191.7 2808.07  1212.9 2826.64  1341.6 2835.52
#Mann= 3 ,-1,0
       0      .1       0   774.9    .045       0   837.9      .1       0
Bank Sta=774.9,837.9
XS Rating Curve= 0 ,0
Exp/Cntr(USF)=0,0
Exp/Cntr=0.3,0.1

Type RM Length L Ch R = 1 ,172470  ,208.2,200.8,198.2
BEGIN DESCRIPTION:
Structure XS 1
END DESCRIPTION:
XS GIS Cut Line= 4
 2320596.2997572653969.5370056692320957.21931898653950.533399782
2321415.05813809654147.2106389792321879.34539128653947.309182746
#Sta/Elev= 30
       0 2962.24      68 2915.07      88 2895.11   136.1 2877.14   188.1 2847.43
   292.3  2814.9   340.3 2808.14   386.4  2771.8   405.3 2770.52   429.9 2789.44
   478.4  2782.7   608.4 2719.96   629.1 2718.18   636.7 2717.41     725 2718.24
   764.6 2756.46   786.9 2770.61   803.9 2774.53   825.5 2761.55   846.8 2761.38
   900.1 2791.51   983.9 2817.48  1052.6 2820.93  1135.3 2833.63  1218.3 2773.92
  1235.5 2774.88  1248.5 2781.85    1320 2835.77    1353    2841  1365.2 2834.05
#Mann= 5 ,-1,0
       0      .1       0   629.1    .045       0     725      .1       0
 1279.71     .12       0 1359.71      .1       0
Bank Sta=629.1,725
XS Rating Curve= 0 ,0
Exp/Cntr(USF)=0,0
Exp/Cntr=0.3,0.1

Type RM Length L Ch R = 1 ,172269  ,566.7,499.8,420.8
BEGIN DESCRIPTION:
Structure XS 4
END DESCRIPTION:
XS GIS Cut Line= 4
2320589.65857687654289.0761885642320850.82015679654176.228592303
2321305.43475887654285.851971528 2321908.3633446 653992.44822125
#Sta/Elev= 30
       0 2963.45    59.6 2928.24   190.1 2870.34   314.7 2767.07   339.4 2767.09
   368.2 2797.19   392.9 2796.79   425.8 2785.47   450.5 2761.26   471.1 2752.46
   516.3 2720.21     541 2714.93   619.2    2715   660.3 2721.28   680.9 2735.31
   742.6 2738.25     773 2757.43   865.4  2759.9   889.4 2778.57   991.1 2803.15
  1055.3 2804.76  1173.3 2826.56  1208.9 2825.82  1235.6 2799.78  1266.8 2777.11
  1287.3  2775.8  1326.2 2800.57  1383.1 2846.36  1397.9 2847.05  1422.7 2833.56
#Mann= 4 ,-1,0
       0      .1       0     541    .045       0   619.2      .1       0
 1312.14     .12       0
Bank Sta=541,619.2
XS Rating Curve= 0 ,0
Exp/Cntr(USF)=0,0
Exp/Cntr=0.3,0.1

Type RM Length L Ch R = 1 ,171770  ,152,150.4,146.9
BEGIN DESCRIPTION:
Structure XS 3
END DESCRIPTION:
XS GIS Cut Line= 5
2321082.14998923655229.7205005492321090.99557781655209.817926253
2321382.90000082654783.0182774522321303.28970364 654300.93370005
2321944.59487541654013.452071324
#Sta/Elev= 30
       0  3065.8    66.2 3016.58    90.4    3010   138.9 2977.29   257.7 2919.68
   319.5 2876.15   371.5 2853.33     449 2809.35   512.3 2762.67   538.9 2752.33
   589.4 2750.16   666.4 2716.14   702.42708.566     752 2706.93   775.9 2708.15
    1023 2739.58  1055.2 2756.77  1146.8 2760.08  1164.2 2765.74  1185.3 2782.97
  1276.1 2802.25  1442.6 2821.14  1493.1 2824.46  1519.4  2797.4  1545.1 2779.37
    1572 2776.08  1668.4 2846.96  1681.6 2849.25  1703.5 2834.58  1730.3 2832.59
#Mann= 6 ,-1,0
       0      .1       0  688.85    .025       0   702.4    .045       0
   775.9    .025       0  888.85      .1       0 1647.47     .12       0
Bank Sta=702.4,775.9
XS Rating Curve= 0 ,0
Exp/Cntr(USF)=0,0
Exp/Cntr=0.3,0.1

Type RM Length L Ch R = 1 ,171619  ,924.3,988.3,1034.9
BEGIN DESCRIPTION:
Structure XS 2
END DESCRIPTION:
XS GIS Cut Line= 4
2321157.33749213655267.3142519982321533.27500662654732.156143139
2321449.24191514654342.9502457872321962.28605256654108.542148518
#Sta/Elev= 30
       0 3098.74    32.3 3078.52    58.1 3043.45    92.6 3018.23   121.3 3006.56
   171.9 2969.25   401.6 2824.39   428.5 2802.84   515.9 2754.72   535.4 2749.23
   615.2  2747.6     654  2725.8   714.3 2714.53     755 2715.42   824.8  2705.3
   882.1 2703.84   886.1 2705.43   947.6 2723.82   976.2 2749.06  1004.9 2760.43
    1073 2779.12  1179.5 2790.03  1231.3 2808.01  1354.5  2799.6  1410.8 2815.69
  1460.7 2779.02    1482 2777.03  1583.1 2846.82  1596.3 2846.13  1616.2 2833.14
#Mann= 5 ,-1,0
       0      .1       0  754.01    .025       0   824.8    .045       0
   886.1      .1       0 1552.18     .12       0
Bank Sta=824.8,886.1
XS Rating Curve= 0 ,0
Exp/Cntr(USF)=0,0
Exp/Cntr=0.3,0.1

Type RM Length L Ch R = 1 ,170631  ,492,469.3,452.1
BEGIN DESCRIPTION:
Structure XS 1
END DESCRIPTION:
XS GIS Cut Line= 4
2321396.16838369655435.3804349452321732.30074958655174.435571948
 2322355.9147442655187.7039548122322523.98092715 655077.13409761
#Sta/Elev= 30
       0 3109.28    35.5 3092.04    60.8 3063.16   111.4 3028.22   136.7 3021.58
   164.1 2999.41   268.4  2936.9   286.7 2920.78   303.8 2887.29   359.5 2848.16
   380.7 2805.89   429.4 2766.67   445.4 2743.86   477.4 2739.68   512.5  2716.7
   541.4 2704.88   585.4 2697.23   653.5 2697.37   732.82689.992   785.5 2689.31
   793.5 2690.38   805.5 2691.11   857.5 2729.34   901.5 2744.34   965.5 2751.66
  1005.5 2768.71  1102.3 2791.99  1175.5 2787.92    1222 2808.54  1250.5 2829.12
#Mann= 7 ,-1,0
       0      .1       0     340     .05       0     390      .1       0
  695.53    .025       0   732.8    .045       0   793.5    .025       0
  795.53      .1       0
Bank Sta=732.8,793.5
XS Rating Curve= 0 ,0
Exp/Cntr(USF)=0,0
Exp/Cntr=0.3,0.1

Type RM Length L Ch R = 1 ,170162  ,505,504.6,503.3
XS GIS Cut Line= 2
2321758.83751531656014.7664866852322577.05445861655249.623074846
#Sta/Elev= 30
       0 2982.41   101.9 2915.69   166.1 2866.23   193.5 2857.28     303  2808.8
     353 2798.82   377.1 2775.72   429.4  2738.8   467.3 2730.95   505.8 2697.28
   523.5 2685.39   536.9 2681.07   573.7 2678.76   585.1 2681.17   613.4 2683.84
   626.1 2690.25   664.5  2692.5   708.3 2687.21   723.7 2705.49   740.2 2717.06
     774 2730.32     786 2738.15     889 2777.88   932.8 2803.59     953 2805.65
  1021.3 2799.98  1036.9 2801.53  1088.8 2790.19  1109.2 2790.39  1120.2 2795.67
#Mann= 6 ,-1,0
       0      .1       0     430     .05       0     470    .025       0
   536.9    .045       0   585.1    .025       0     600      .1       0
Bank Sta=536.9,585.1
XS Rating Curve= 0 ,0
Exp/Cntr(USF)=0,0
Exp/Cntr=0.3,0.1

Type RM Length L Ch R = 1 ,169657  ,419.5,422.8,426.7
XS GIS Cut Line= 2
2322183.42576697656390.7040011732322930.87800165655497.299554979
#Sta/Elev= 30
       0 2989.77    38.5 2963.94    64.6 2954.78   115.2 2915.72   169.5 2866.19
   210.6  2841.6   226.2 2836.73   265.7 2816.35   346.2 2762.34   376.4 2748.28
   403.6 2741.48   440.1 2725.96   467.3 2723.31   518.4  2691.3   549.7 2678.77
   595.1 2672.62   666.1 2672.08   671.8 2672.62   695.6 2674.43   705.6  2678.3
   722.9 2691.34   755.4 2708.77   794.7 2741.31     946  2762.7   995.8 2776.64
  1060.8 2786.52  1080.7 2795.87  1114.7  2797.4    1146 2814.55  1164.8 2817.35
#Mann= 3 ,-1,0
       0      .1       0   595.1    .045       0   671.8      .1       0
Bank Sta=595.1,671.8
XS Rating Curve= 0 ,0
Exp/Cntr(USF)=0,0
Exp/Cntr=0.3,0.1

Type RM Length L Ch R = 1 ,169234  ,467.5,482.5,491.4
XS GIS Cut Line= 2
2322515.13533857656607.4209212892323282.01161637655766.074454814
#Sta/Elev= 30
       0 3004.63    19.4 2992.78      49 2965.18    73.4  2956.2   114.4 2921.79
   126.2 2909.34     160 2885.11   376.5 2736.41   392.7 2719.67   410.1 2719.41
   424.2  2715.7   452.8 2692.91   486.5 2676.86   514.8 2673.87   538.9 2673.92
   582.1 2668.89     685 2668.89   708.2 2678.41   717.5 2684.55   744.5 2708.09
   755.3 2714.12     815 2732.23   877.2 2757.09   939.5  2776.3  1036.8 2792.86
  1058.4 2801.24  1096.3  2803.8    1106 2806.41    1118 2812.56  1138.4 2813.23
#Mann= 6 ,-1,0
       0      .1       0     540    .025       0   582.1    .045       0
     685      .1       0     700     .12       0     800      .1       0
Bank Sta=582.1,685
XS Rating Curve= 0 ,0
Exp/Cntr(USF)=0,0
Exp/Cntr=0.3,0.1

Type RM Length L Ch R = 1 ,168752  ,297.1,308.4,311.8
XS GIS Cut Line= 4
2322656.66475579656775.487104237 2323063.5618303656625.112098442
2323527.95523055656311.093703987 2323745.6877024656088.759109289
#Sta/Elev= 30
       0 2935.17     122 2884.78   213.1 2837.89   242.5 2828.38   269.2 2814.17
   289.5 2812.09   306.6 2805.79   383.3  2754.7   454.4 2720.44   463.5 2713.22
   497.3 2709.88   521.5 2695.51   569.7 2686.35   627.2 2660.98   726.5 2660.84
   776.4 2668.07   801.5  2682.2     824 2699.64   890.7 2724.61     956 2724.11
   987.3 2727.27    1027 2746.87  1083.6 2763.24  1137.3 2769.17  1177.6 2780.69
  1200.5 2791.25  1227.8 2809.38  1250.5 2810.98    1277 2804.83  1305.6 2810.84
#Mann= 5 ,-1,0
       0      .1       0   627.2    .045       0   726.5      .1       0
 1134.39     .06       0 1274.39      .1       0
Bank Sta=627.2,726.5
XS Rating Curve= 0 ,0
Exp/Cntr(USF)=0,0
Exp/Cntr=0.3,0.1

Type RM Length L Ch R = 1 ,168443  ,465.4,462.3,454.3
XS GIS Cut Line= 2
 2322727.4294644657018.740790082 2324027.7309851656510.119446951
#Sta/Elev= 30
       0 2987.44    30.9 2965.37    56.6 2961.74   219.9 2853.36   297.2 2817.71
   358.3 2777.22   374.5 2771.46   403.1 2752.13   461.8 2726.73   495.8 2717.79
   511.2 2709.12   533.4 2707.43   588.4 2689.52   623.6 2671.34   684.1  2668.5
   722.4 2654.84   773.9 2654.38   786.8 2654.75   842.6 2661.42   894.2 2702.09
   932.8 2722.19   948.6 2725.79  1074.6 2728.12    1141 2753.84  1207.7  2762.9
  1250.7 2775.75  1295.4 2795.85  1343.9 2804.93  1375.2 2821.67  1396.2 2822.19
#Mann= 3 ,-1,0
       0      .1       0   722.4    .045       0   786.8      .1       0
Bank Sta=722.4,786.8
XS Rating Curve= 0 ,0
Exp/Cntr(USF)=0,0
Exp/Cntr=0.3,0.1

Type RM Length L Ch R = 1 ,167981  ,528.5,508.4,486.1
XS GIS Cut Line= 2
2322921.18180269657545.1378017962324069.57759863656893.116458066
#Sta/Elev= 30
       0 2971.23    26.4 2969.47    44.8 2959.44   136.8 2893.42   207.5 2851.39
   270.2 2804.79     307 2784.37   320.8 2779.42   396.9 2772.71   449.6 2760.99
   515.6 2729.66   544.9 2703.19   574.3 2698.44   623.7 2662.58     698 2650.18
   702.6 2650.09   771.6 2650.16     790 2660.18   817.6 2690.65   872.8  2711.9
   900.4 2713.87   918.8 2722.41   937.2 2718.71   964.8 2726.41   992.4 2719.19
  1034.9 2728.93  1084.4  2748.6  1161.1 2759.18  1245.4 2788.43  1320.6  2795.6
#Mann= 3 ,-1,0
       0      .1       0     698    .045       0   771.6      .1       0
Bank Sta=698,771.6
XS Rating Curve= 0 ,0
Exp/Cntr(USF)=0,0
Exp/Cntr=0.3,0.1

Type RM Length L Ch R = 1 ,167473  ,563.3,547.1,531.2
XS GIS Cut Line= 2
2323519.10964197658142.1305392572324244.44790522657018.740790082
#Sta/Elev= 30
       0 2939.69    44.9 2928.67   177.9 2879.57   215.4 2869.64   258.2 2862.47
   304.3 2846.22   329.7 2832.17   372.5 2796.16   467.7 2738.89   496.3 2727.75
     563 2709.55   588.8 2694.57   611.9 2688.84   652.4 2657.65   677.2 2645.37
   788.4 2645.28   805.8 2645.28   824.8 2650.84   839.1 2667.05   846.3 2672.29
   877.2 2684.99   910.5 2691.91   967.7 2694.59  1002.5 2699.67    1082 2722.13
  1134.3 2749.68  1161.7 2759.68  1210.8 2769.91  1277.2 2775.32  1337.2 2793.82
#Mann= 6 ,-1,0
       0      .1       0     540     .05       0     650      .1       0
     660     .05       0   677.2    .045       0   805.8      .1       0
Bank Sta=677.2,805.8
XS Rating Curve= 0 ,0
Exp/Cntr(USF)=0,0
Exp/Cntr=0.3,0.1

Type RM Length L Ch R = 1 ,166926  ,589.4,574.3,562.7
XS GIS Cut Line= 2
2324186.95157947658540.1820251852324598.27144826657085.082704403
#Sta/Elev= 30
       0 2941.31    31.6 2924.97    48.8 2907.57    69.6 2900.06   102.9 2872.86
     159 2844.93   223.8 2831.23   360.6 2788.72   460.4 2771.06   593.4 2727.64
   626.6 2710.17   655.7 2685.65     689 2681.46   729.3  2643.6   747.2 2638.16
   754.5 2638.03   846.9 2638.04   886.8 2654.56   938.4 2653.94   984.1 2673.42
    1088 2707.25    1113 2713.67  1146.2 2714.13  1204.4 2733.86  1244.6 2737.85
  1320.8 2729.71  1416.4 2738.75  1466.3 2756.49  1499.5 2780.58  1512.1 2784.18
#Mann= 4 ,-1,0
       0      .1       0     680    .025       0   747.2    .045       0
   846.9      .1       0
Bank Sta=747.2,846.9
XS Rating Curve= 0 ,0
Exp/Cntr(USF)=0,0
Exp/Cntr=0.3,0.1

Type RM Length L Ch R = 1 ,166351  ,868.4,883.2,894.1
XS GIS Cut Line= 2
2324969.78616846658540.1820251852324983.05455133657142.579030148
#Sta/Elev= 30
       0 2919.33      99 2886.55     143 2866.97     159 2854.81     183  2854.2
   222.7  2829.8     247 2821.96     299  2798.1     371 2770.12     427 2750.88
     519 2727.94     563 2709.32     575 2696.63     611 2676.53     635 2673.36
     679 2648.26     735 2625.43     831 2625.41     859  2640.1     887 2663.28
     899  2667.7     911 2676.53     927 2683.81     979 2699.16  1026.4 2706.84
  1115.3 2715.02  1199.1  2733.4  1228.3 2744.54  1261.5 2751.52  1397.7 2770.15
#Mann= 3 ,-1,0
       0      .1       0     735    .045       0     831      .1       0
Bank Sta=735,831
XS Rating Curve= 0 ,0
Exp/Cntr(USF)=0,0
Exp/Cntr=0.3,0.1

Type RM Length L Ch R = 1 ,165468  ,632.7,655.1,683.2
XS GIS Cut Line= 3
2325199.77147144658624.2151166592325650.89648883658208.472453578
2326017.98841474657328.336390248
#Sta/Elev= 30
       0 2889.67    45.8 2863.45    70.4 2843.12    87.1 2838.36   138.3 2806.87
   194.9  2779.6   354.1 2725.74   488.5 2686.71   582.7 2664.94   605.4 2664.72
   669.1 2650.94   687.3 2652.91   725.4 2644.04   946.4 2643.89   965.6 2635.73
  1007.1    2632  1063.6 2614.09  1133.8 2614.21  1158.8 2621.34  1184.8  2643.3
  1213.4 2657.71  1280.1 2706.41    1302 2744.33  1319.2 2762.86  1336.5 2774.48
  1423.2 2816.03    1455 2826.98  1483.8 2845.55  1522.3 2848.76  1567.1 2867.93
#Mann= 5 ,-1,0
       0      .1       0  1063.6    .045       0  1133.8    .025       0
 1183.48      .1       0 1393.48     .06       0
Bank Sta=1063.6,1133.8
XS Rating Curve= 0 ,0
Exp/Cntr(USF)=0,0
Exp/Cntr=0.3,0.1

Type RM Length L Ch R = 1 ,164813  ,599.1,593.6,588.9
XS GIS Cut Line= 4
2325491.67589446659017.8438082992325898.57296896658456.148933711
 2326517.7641693658093.4798020882326641.60240936657872.340087683
#Sta/Elev= 30
       0 2900.04    46.7  2878.5   124.3  2824.6   144.1 2818.65   184.1 2791.86
   272.9 2759.32   389.5 2732.83   440.4 2711.59   509.6 2688.87   590.9 2673.29
   623.2 2672.19   648.6  2660.1   677.5  2661.6   774.3 2639.72   806.7 2635.55
   875.3 2637.26     918  2634.2   964.3 2638.47  1043.1  2638.2  1052.4 2635.45
  1071.4 2615.38  1088.7 2606.68  1186.8 2606.55  1205.4 2611.14    1312 2617.53
  1380.1 2634.46  1457.4 2675.96  1538.9 2739.55  1617.8 2793.37  1664.6 2810.38
#Mann= 5 ,-1,0
       0      .1       0     670     .12       0  853.59      .1       0
  1088.7    .045       0  1186.8      .1       0
Bank Sta=1088.7,1186.8
XS Rating Curve= 0 ,0
Exp/Cntr(USF)=0,0
Exp/Cntr=0.3,0.1

Type RM Length L Ch R = 1 ,164219  ,687,681.8,684.1
XS GIS Cut Line= 4
2325978.18326615659407.049705651 2326367.3891635658911.696745385
2326946.77521524658447.3033451352327088.30463246658186.358482138
#Sta/Elev= 30
       0 2914.91    51.2 2888.76   180.4 2807.02   223.4 2795.88   239.2  2786.4
   262.2 2786.38   378.7 2738.05   441.5 2722.06   516.2 2690.87   541.6 2675.35
   563.9 2666.13   582.3 2650.01   612.8 2647.94   636.1 2634.74   680.7 2627.05
   723.2 2625.79   779.6 2629.44   800.1 2622.01   838.7  2616.7   856.5 2606.56
   870.6 2603.42   943.7 2603.38   985.2 2608.89  1107.7 2611.88    1184 2622.71
  1218.5 2635.99  1289.6  2648.5  1506.9 2723.23  1602.4 2764.64  1669.3 2782.51
#Mann= 5 ,-1,0
       0      .1       0   870.6    .045       0   943.7      .1       0
  959.96    .025       0 1009.96      .1       0
Bank Sta=870.6,943.7
XS Rating Curve= 0 ,0
Exp/Cntr(USF)=0,0
Exp/Cntr=0.3,0.1

Type RM Length L Ch R = 1 ,163538  ,716.3,725.6,746.7
XS GIS Cut Line= 3
2326526.60975787659769.7188372742327375.78626119658880.737185368
2327716.34142137658770.167328166
#Sta/Elev= 30
       0 2959.06    22.9 2947.79      37 2936.84    77.5 2895.74   181.8 2822.96
   244.8 2791.89   297.6 2754.09   312.7 2750.79   369.3 2710.89   487.5 2651.14
   505.1 2638.96   533.4 2636.77   559.4 2616.95     590 2603.05     674 2609.37
     703 2604.97   785.2 2605.05     825 2596.69   830.4    2596   937.9  2596.9
   969.1 2621.21   979.9 2625.03    1091 2628.18  1134.7 2639.86  1178.4 2641.99
  1280.1 2678.63  1406.4 2706.09    1477 2726.95  1553.6 2739.05  1587.4 2737.85
#Mann= 3 ,-1,0
       0      .1       0     825    .045       0   937.9      .1       0
Bank Sta=825,937.9
XS Rating Curve= 0 ,0
Exp/Cntr(USF)=0,0
Exp/Cntr=0.3,0.1

Type RM Length L Ch R = 1 ,162812  ,487.9,483.6,477.6
XS GIS Cut Line= 2
2326973.31198097 660127.965174612328304.57306168659168.218814094
#Sta/Elev= 30
       0 2881.44    52.8 2845.81   200.8 2754.56   227.5 2735.43   236.1  2725.7
   250.1 2721.33   313.5 2680.96   365.1 2657.33   412.8  2640.8   427.6 2628.91
   459.8 2625.87   521.3 2588.83   526.2 2588.63   590.3 2588.83   640.9 2594.83
   664.3 2604.12   729.8 2610.04   792.5 2606.86   852.2 2613.51  1078.5 2614.94
  1182.1 2624.93  1211.7 2624.36  1295.5 2634.18  1394.1 2637.86  1418.8 2640.62
  1487.8 2657.03  1514.1 2651.39  1564.3 2650.72    1619 2674.38  1641.1 2678.85
#Mann= 7 ,-1,0
       0      .1       0   521.3    .045       0   590.3      .1       0
     790     .12       0     980      .1       0    1140     .12       0
    1150      .1       0
Bank Sta=521.3,590.3
XS Rating Curve= 0 ,0
Exp/Cntr(USF)=0,0
Exp/Cntr=0.3,0.1

Type RM Length L Ch R = 1 ,162328  ,603.6,626.9,642.4
BEGIN DESCRIPTION:
Structure XS 4
END DESCRIPTION:
XS GIS Cut Line= 3
2327181.18331251660402.1784204712327565.96641557660326.990917574
 2328596.4774847659358.398968482
#Sta/Elev= 30
       0 2840.23    88.6 2785.94   194.3 2705.96   210.9 2698.53   223.1 2696.64
   251.7 2677.54   312.8 2643.91   345.4 2621.67   400.6    2618   437.4 2602.34
   533.6 2599.95   547.7 2587.02   564.7  2582.2   680.9 2582.28     726 2589.93
   748.6 2601.51   799.6 2598.97   834.3 2604.87   902.8 2602.67   938.6 2608.02
  1034.4  2606.5  1354.2 2615.09  1393.4 2625.68  1413.6 2626.31  1422.1  2630.7
  1438.1 2631.86    1504 2647.43  1583.4 2671.17  1648.5 2685.88  1806.3 2710.11
#Mann= 5 ,-1,0
       0      .1       0   564.7    .045       0   680.9      .1       0
  942.06     .12       0 1132.06      .1       0
Bank Sta=564.7,680.9
XS Rating Curve= 0 ,0
Exp/Cntr(USF)=0,0
Exp/Cntr=0.3,0.1

Type RM Length L Ch R = 1 ,161701  ,131,128.9,127.8
BEGIN DESCRIPTION:
Structure XS 3
END DESCRIPTION:
XS GIS Cut Line= 4
2327256.37081541660671.9688720452327884.40760432660716.196814926
2328565.51792468660477.3659233692328998.95176492660671.968872045
#Sta/Elev= 30
       0  2795.2    31.9 2774.03      68 2756.19      72 2752.43      84 2726.86
   164.2 2678.19   180.2  2676.5   264.5 2641.12   324.6  2624.3   336.6 2616.35
   360.7 2613.97   384.8 2597.63   396.8 2593.27   420.8 2590.48   650.4 2595.22
   744.8 2586.83   798.9  2588.7   862.5 2583.13   878.9 2576.66   968.4  2576.2
  976.172576.811  1002.4 2585.04  1023.6 2603.34  1174.7 2610.59  1507.6 2640.84
    1534 2658.17  1568.1 2659.06  1621.7 2679.05  1709.4 2699.37  1826.5 2742.43
#Mann= 11 ,-1,0
       0      .1       0     550     .06       0  649.59     .07       0
  759.59     .06       0  859.59     .07       0   878.9    .045       0
  976.17      .1       0 1069.59     .08       0 1149.59      .1       0
 1381.36     .06       0 1711.36      .1       0
Bank Sta=878.9,976.17
XS Rating Curve= 0 ,0
Exp/Cntr(USF)=0,0
Exp/Cntr=0.3,0.1

Type RM Length L Ch R = 1 ,161572  ,578.1,589,599.7
BEGIN DESCRIPTION:
Structure XS 2
END DESCRIPTION:
XS GIS Cut Line= 4
2327190.02890109660831.1894664162327919.78995862660840.035054992
2328587.63189612660601.2041634352328998.95176491660751.579169231
#Sta/Elev= 30
       0 2811.04    46.1 2789.11   158.2 2716.66   250.2 2668.23   270.2 2664.15
   350.2 2634.41   390.2 2613.81   410.2 2612.56   430.2 2600.39   450.2 2593.86
   534.2 2589.91   754.3 2594.47     777 2590.29   827.9 2590.71   857.7 2585.31
   960.8 2584.55  1014.8 2575.04  1015.82575.042  1094.7 2575.16  1108.3 2595.02
    1121 2602.27  1218.8 2605.79  1442.6 2625.46  1461.3 2629.94  1501.9 2648.07
  1575.9 2666.46  1601.5 2667.23  1614.1 2673.55  1695.2 2691.12    1877 2756.05
#Mann= 12 ,-1,0
       0      .1       0     520     .06       0     620     .07       0
     700     .06       0  739.81     .07       0  929.81     .06       0
  1015.8    .045       0  1094.7     .07       0 1129.81     .08       0
 1239.81     .07       0 1339.81     .06       0 1659.08      .1       0
Bank Sta=1015.8,1094.7
XS Rating Curve= 0 ,0
Exp/Cntr(USF)=0,0
Exp/Cntr=0.3,0.1

Type RM Length L Ch R = 1 ,160983  ,807.6,825.1,849.4
BEGIN DESCRIPTION:
Structure XS 1
END DESCRIPTION:
XS GIS Cut Line= 4
2327097.15022104 661215.972569482327393.47743834661384.038752428
2328472.63924463661300.0056609542328981.26058776661392.884341004
#Sta/Elev= 30
       0 2758.81    72.5 2723.52   132.2 2687.31   219.6 2658.92   246.7 2648.57
   258.4  2639.8   278.9 2641.54   325.4 2605.32   351.4 2603.42   383.5 2587.25
   628.2  2583.4   688.4 2587.28   965.3 2587.79    1001 2580.96  1157.8 2580.42
  1193.9 2568.76  1246.1 2568.68  1284.6 2574.56  1374.5 2573.49  1394.5 2585.86
  1418.6 2607.98  1479.6 2641.83  1512.1 2669.35  1528.3 2672.81  1545.4 2687.84
  1605.6 2716.17    1635 2718.43  1666.6 2728.55  1760.1  2742.7  1940.1 2780.86
#Mann= 11 ,-1,0
       0      .1       0  360.67     .06       0 1150.67      .1       0
  1193.9    .045       0  1246.1      .1       0 1250.67    .025       0
 1350.67      .1       0  1553.1     .06       0  1603.1      .1       0
  1653.1     .06       0  1853.1      .1       0
Bank Sta=1193.9,1246.1
XS Rating Curve= 0 ,0
Exp/Cntr(USF)=0,0
Exp/Cntr=0.3,0.1

Type RM Length L Ch R = 1 ,160158  ,601,607.4,614.4
XS GIS Cut Line= 2
2327016.88302922661505.2474837592328711.47013619662348.207907231
#Sta/Elev= 30
       0 2731.72   110.9 2675.31   204.7 2640.47   226.2 2625.49   240.5 2621.97
   260.3 2609.97   288.8 2600.24   311.9 2599.26   339.5 2583.85   888.3 2577.92
   941.9 2580.13  1008.9 2577.53  1053.6 2570.82  1122.5 2573.16  1183.1 2568.15
  1330.5 2573.96  1365.8 2562.55  1440.4 2562.37  1449.4 2562.47  1473.3 2573.97
  1529.9 2627.11  1607.5 2672.22  1631.4 2689.86  1714.8 2729.68  1781.8 2767.45
  1799.6 2781.99  1825.3 2785.41  1867.9 2811.49  1884.5 2826.97  1892.7 2829.52
#Mann= 13 ,-1,0
       0      .1       0     220     .06       0     280     .07       0
     330     .06       0     500     .07       0     550     .06       0
     660     .07       0     720     .06       0     940     .07       0
     990     .06       0    1210      .1       0  1365.8    .045       0
  1449.4      .1       0
Bank Sta=1365.8,1449.4
XS Rating Curve= 0 ,0
Exp/Cntr(USF)=0,0
Exp/Cntr=0.3,0.1

Type RM Length L Ch R = 1 ,159551  ,854.3,842.5,692.1
XS GIS Cut Line= 4
2326885.99248613 661788.008080682327017.53992385661972.270392744
2328123.23849587662759.5277760242328609.74586756662640.112330245
#Sta/Elev= 30
       0 2701.89    11.3 2700.05   104.6 2662.23   175.9 2629.69   197.4  2618.7
   210.3 2607.04   240.4 2593.85   296.9 2597.58   469.9 2589.58   509.5 2593.45
   543.9 2586.15   671.6    2580   772.8 2580.87  1231.3  2567.2  1276.2 2569.74
  1319.7  2565.9  1338.9 2557.19  1345.2    2557  1436.4 2557.25    1467 2564.01
  1517.6 2586.45  1583.7 2599.41  1621.8 2622.57  1660.7 2654.41  1757.7 2700.11
  1778.3 2704.15  1864.8 2767.09  1897.7 2781.66  1956.8 2799.35  2084.7 2819.15
#Mann= 12 ,-1,0
       0      .1       0   346.4     .07       0   476.4     .06       0
   996.4     .08       0  1076.4     .06       0  1166.4     .08       0
  1316.4     .05       0  1336.4      .1       0  1338.9    .045       0
  1436.4      .1       0  1436.4    .025       0  1506.4      .1       0
#XS Ineff= 2 , 0
         1274.37 2591.38
Permanent Ineff=
       F       F
Bank Sta=1338.9,1436.4
XS Rating Curve= 0 ,0
Exp/Cntr(USF)=0,0
Exp/Cntr=0.3,0.1

Type RM Length L Ch R = 1 ,158709  ,547.4,550.7,540.8
XS GIS Cut Line= 4
2326853.89653519663480.443244983 2327331.5583183663338.913827764
2328008.24584438663356.605004916 2328260.3451188663414.101330661
#Sta/Elev= 30
       0 2691.78    69.7 2680.33   173.4  2645.7   215.1 2639.79   290.2 2618.44
   348.6 2599.94     484 2584.58   542.8 2570.17   578.7 2576.19   594.8 2573.47
   618.8 2556.57   650.9 2555.96  666.932545.299   674.9 2541.97   706.9 2542.16
   714.9 2550.94   878.9 2560.87     971  2556.8     995 2549.89  1054.7 2545.33
    1063 2559.64    1071 2566.17    1127 2564.88    1159 2573.52  1179.1 2589.84
  1220.2 2607.78  1322.7 2682.73    1372 2706.32  1392.5 2706.99  1433.7 2727.13
#Mann= 9 ,-1,0
       0      .1       0   173.4     .06       0   290.2      .1       0
     484     .12       0   578.7      .1       0  666.93    .045       0
   714.9     .08       0     995    .045       0  1054.7      .1       0
Bank Sta=666.93,1054.7
XS Rating Curve= 0 ,0
Exp/Cntr(USF)=0,0
Exp/Cntr=0.3,0.1

Type RM Length L Ch R = 1 ,158158  ,525.4,527.2,530.8
XS GIS Cut Line= 3
 2326889.2788895663807.7300223012327278.48478685663714.851342251
2328043.62819869663966.950616673
#Sta/Elev= 30
       0 2713.95   153.9 2665.85   179.8 2654.21   204.5  2653.5   230.3 2638.64
   253.8 2637.44   274.4 2627.46   286.7 2626.25   315.5 2613.64   469.8 2566.74
   524.8 2561.67   557.7 2570.37   604.1 2555.19   646.2 2554.74   688.3 2547.71
     722 2550.42   747.3 2543.68   797.8 2537.89   840.5 2537.76   843.6 2537.88
     855 2544.82   873.6 2567.16   903.8 2597.72   924.1 2612.62   978.9 2641.34
  1037.9 2676.68  1092.6 2686.86  1130.5 2702.18  1147.7 2712.59  1205.7 2734.93
#Mann= 5 ,-1,0
       0      .1       0     140     .06       0     240      .1       0
   797.8    .045       0   843.6      .1       0
Bank Sta=797.8,843.6
XS Rating Curve= 0 ,0
Exp/Cntr(USF)=0,0
Exp/Cntr=0.3,0.1

Type RM Length L Ch R = 1 ,157631  ,452.9,444.8,436.6
XS GIS Cut Line= 4
2326787.55462087 664157.130771062327128.10978105664165.976359637
2327610.19435845664395.9616626172327862.29363288664400.384456906
#Sta/Elev= 30
       0 2797.75    12.6 2796.05    96.7 2751.26   120.7 2735.08   204.7 2695.89
   224.7 2678.01   256.7 2674.28   272.7 2661.64   288.7 2635.49   358.5 2588.54
   373.1 2586.94   391.1 2576.64   424.9  2567.9     487 2559.23   515.3 2562.39
   543.2  2548.5   589.2 2548.87   664.5  2533.6   668.7 2533.39   730.2  2533.5
   747.6 2539.69   761.8 2558.96   783.9 2582.17   806.1  2599.9   871.2 2600.15
     957 2645.23  1028.8  2668.9  1040.8 2669.72  1060.8 2682.87  1126.9 2690.85
#Mann= 5 ,-1,0
       0      .1       0     230     .06       0     330      .1       0
   664.5    .045       0   730.2      .1       0
Bank Sta=664.5,730.2
XS Rating Curve= 0 ,0
Exp/Cntr(USF)=0,0
Exp/Cntr=0.3,0.1

Type RM Length L Ch R = 1 ,157186  ,445,428,398.1
XS GIS Cut Line= 2
2326654.87079223664564.0278455652327760.56936425664824.972708562
#Sta/Elev= 30
       0 2778.74      26 2767.57      63 2745.15     100 2718.46   131.7 2701.49
   161.6 2699.16   181.6 2685.82   256.2 2657.06   268.5 2654.57   314.6 2625.39
   330.1  2623.7   403.7 2588.46   453.4  2556.7   478.1 2555.81     511 2538.66
   544.9 2529.55     548 2529.33   617.2 2529.62   646.6 2536.72     677 2558.92
   713.6 2567.98   757.6  2590.5   776.8 2595.59   843.9 2594.52   864.4 2600.75
   901.4  2618.1   913.1 2619.36     963 2637.02  1049.9 2655.95  1136.1  2665.8
#Mann= 5 ,-1,0
       0      .1       0      70     .06       0     280      .1       0
   544.9    .045       0   617.2      .1       0
Bank Sta=544.9,617.2
XS Rating Curve= 0 ,0
Exp/Cntr(USF)=0,0
Exp/Cntr=0.3,0.1

Type RM Length L Ch R = 1 ,156758  ,469.8,467,461.3
XS GIS Cut Line= 3
2326681.40755796665329.1712574052327473.08773552665019.575657238
2327822.48848428665032.844040103
#Sta/Elev= 30
       0 2732.68    11.6 2731.85    37.3 2708.11    80.3 2680.66    93.2 2675.08
   141.1 2658.33   205.9 2645.25   226.3 2638.82   243.5 2638.64   290.7 2623.18
   350.9 2618.57   376.6 2599.29   398.1 2594.09   415.9 2584.86   434.4 2581.12
   462.5 2552.03   488.3 2548.66   522.7 2526.31   544.1 2526.21   552.7 2523.58
   634.3 2523.63   678.3 2540.67   733.1 2553.66   770.9 2566.65   853.2 2602.88
   897.2 2618.97   993.3 2635.46  1077.3 2660.58  1101.3 2662.49  1199.7 2680.13
#Mann= 4 ,-1,0
       0     .06       0     150      .1       0   552.7    .045       0
   634.3      .1       0
Bank Sta=552.7,634.3
XS Rating Curve= 0 ,0
Exp/Cntr(USF)=0,0
Exp/Cntr=0.3,0.1

Type RM Length L Ch R = 1 ,156291  ,583.4,570.8,546
XS GIS Cut Line= 2
2326906.97006665665793.5646576542327933.05834149665284.943314524
#Sta/Elev= 30
       0 2777.27    10.3 2769.05    19.1 2755.95    37.1 2754.59    93.7 2703.24
   108.9 2693.57   130.8 2689.99   175.5 2658.54     199 2637.31     235 2614.47
   281.8 2595.42   397.2 2564.83   443.3 2540.43   469.8 2541.94     488 2532.91
   511.6 2529.75   541.4 2520.07   581.7  2514.3   635.3 2514.26   662.1 2523.59
   679.9 2538.94   711.2 2559.84   751.4 2563.94   800.5 2577.73   854.1 2610.96
   898.7 2623.99   968.3 2635.66  1032.6 2655.93  1095.1 2667.01  1145.2 2682.03
#Mann= 6 ,-1,0
       0     .06       0     130      .1       0   581.7    .045       0
   635.3      .1       0    1010     .06       0    1120      .1       0
Bank Sta=581.7,635.3
XS Rating Curve= 0 ,0
Exp/Cntr(USF)=0,0
Exp/Cntr=0.3,0.1

Type RM Length L Ch R = 1 ,155720  ,461.9,453.3,451.9
XS GIS Cut Line= 3
2327291.75316971666395.0646808352327645.57671276666125.274229261
2328021.51422725665497.237440352
#Sta/Elev= 30
       0 2688.35     7.4 2684.72    18.8 2673.94    36.1 2673.13    65.9 2651.19
   126.3 2624.07   141.4 2622.44   195.7 2606.48   326.4 2595.46   398.4  2569.4
   412.6 2560.38   426.9 2556.93   438.2 2550.77   458.6 2533.63   484.8 2530.83
   512.3 2510.71   527.9  2506.8     529 2506.75   595.6 2506.89   626.9 2520.51
   640.9 2532.69   674.4 2554.22   770.6 2587.23   855.3 2605.71   986.4 2624.82
  1038.9 2636.81  1073.1 2648.07  1088.5 2648.72  1139.7 2665.67  1176.9 2672.03
#Mann= 5 ,-1,0
       0      .1       0   527.9    .045       0   595.6      .1       0
 1104.95     .06       0 1144.95      .1       0
Bank Sta=527.9,595.6
XS Rating Curve= 0 ,0
Exp/Cntr(USF)=0,0
Exp/Cntr=0.3,0.1

Type RM Length L Ch R = 1 ,155267  ,556.5,584.8,614.7
XS GIS Cut Line= 3
2327535.00685556666589.6676295112327999.40025581666461.406595156
2328322.26423884665713.954360469
#Sta/Elev= 30
       0 2652.63    63.5 2638.98   138.2 2628.91   150.6 2624.71   171.4 2626.57
   221.1 2612.92   316.6 2602.26   358.1 2591.18   424.1 2578.92   508.2 2549.94
   538.7  2526.7     591 2524.58   608.4 2508.57   625.6 2501.56   630.2 2501.28
   699.9 2501.64   821.9 2513.64   878.5 2549.15   891.6 2560.89   945.1 2584.61
  1008.3 2619.36  1036.3 2620.29  1051.6 2629.98  1061.5  2632.7    1092 2633.41
  1118.2 2638.04  1205.3 2666.24  1218.4 2667.18  1260.5 2684.74    1296 2695.54
#Mann= 7 ,-1,0
       0      .1       0   625.6    .045       0   699.9      .1       0
  711.78    .025       0  741.78      .1       0  991.78     .06       0
 1141.78      .1       0
Bank Sta=625.6,699.9
XS Rating Curve= 0 ,0
Exp/Cntr(USF)=0,0
Exp/Cntr=0.3,0.1

Type RM Length L Ch R = 1 ,154682  ,573.3,576.1,584.9
XS GIS Cut Line= 3
2327738.45539281667014.2558811672328684.93337046 666545.43968663
2328950.30102775666218.152909311
#Sta/Elev= 30
       0 2677.57   101.6 2641.84   118.5 2630.56   144.8 2628.62   172.2 2611.32
   269.7 2573.69   366.3 2558.22     417 2542.31   475.1 2529.49   582.2 2515.81
     609 2519.94   635.8  2508.5   733.5 2513.02   796.5 2510.47   814.3 2504.28
   845.6 2499.99   854.5 2495.41   939.3 2495.47   970.6  2520.1   992.9 2548.43
  1002.7 2557.52  1038.8 2581.22  1061.7 2583.22  1093.1 2597.67  1143.9 2597.82
  1195.6 2613.81  1246.4 2642.87  1314.7 2672.81  1405.7 2698.27  1477.6 2710.86
#Mann= 6 ,-1,0
       0      .1       0     830     .12       0   854.5    .045       0
   939.3     .12       0     960     .06       0 1066.22      .1       0
#XS Ineff= 2 , 0
          730.11 2539.48
Permanent Ineff=
       F       F
Bank Sta=854.5,939.3
XS Rating Curve= 0 ,0
Exp/Cntr(USF)=0,0
Exp/Cntr=0.3,0.1

Type RM Length L Ch R = 1 ,154106  ,525.1,525.2,540.6
XS GIS Cut Line= 3
2328034.78261011667474.226487129 2329003.3745592666925.799995405
2329295.27898222666580.822040934
#Sta/Elev= 30
       0    2675    29.2 2669.43    79.7 2647.76   140.1 2628.18   192.6 2626.14
   221.3  2611.4   261.9 2597.03   327.6 2580.86   470.5 2538.29   515.4 2511.38
   534.8 2510.67   562.4 2488.81   617.6 2488.65   619.1 2488.88   663.5 2494.17
   681.9  2500.8   746.3 2501.51   769.2 2495.13   829.4 2495.69   861.2 2504.78
   976.1 2508.09    1090    2533  1114.3 2539.48  1134.9  2552.1  1155.8 2552.13
  1213.4 2586.47  1276.3 2613.45  1454.5 2656.94  1529.2 2688.72    1565 2699.37
#Mann= 5 ,-1,0
       0      .1       0   562.4    .045       0   619.1      .1       0
    1090     .06       0 1223.08      .1       0
Bank Sta=562.4,619.1
XS Rating Curve= 0 ,0
Exp/Cntr(USF)=0,0
Exp/Cntr=0.3,0.1

Type RM Length L Ch R = 1 ,153581  ,537.5,543.7,542.8
XS GIS Cut Line= 2
2328397.45174173667867.8551787692329596.02899381667182.322064115
#Sta/Elev= 30
       0 2678.36    99.9 2646.08   118.3 2644.94   159.8  2629.3   267.8 2601.36
   279.3  2595.1   291.2 2596.05   341.1 2579.03   399.7 2553.47   414.4 2542.19
   450.1 2503.27   467.1  2501.8   505.4 2486.66   633.8 2486.35  636.292486.766
   657.5 2490.87   671.3 2499.22   780.8 2499.76   841.8 2511.36   906.8 2514.03
   966.2 2532.71  1003.1 2533.06  1021.5 2540.95  1076.9 2550.29  1101.1  2558.8
  1132.1 2578.54  1246.1 2630.04    1298 2645.19  1348.7 2667.98  1380.8 2677.02
#Mann= 6 ,-1,0
       0      .1       0     480    .025       0   505.4    .045       0
  636.29      .1       0     910     .07       0    1020      .1       0
Bank Sta=505.4,636.29
XS Rating Curve= 0 ,0
Exp/Cntr(USF)=0,0
Exp/Cntr=0.3,0.1
